HEC-RAS study LLRiver.prj: LLRiver

--- LLRiver.g01 (geometry) --- (continued)

Type RM Length L Ch R = 1 ,63698.22,633.17,633.17,736.74
XS GIS Cut Line= 2
  1343966.703731   795799.884915  1343119.481458   795897.107059
#Sta/Elev= 30
       0 1089.35   39.08 1083.91   68.66  1078.4   83.32 1078.67  113.91  1077.7
  124.73 1074.78  136.72 1073.83  164.02 1070.02  218.91 1065.43  253.48 1063.69
  343.12 1049.57  371.03  1045.9  396.68  1044.3  418.93 1043.98  436.24 1044.02
  450.54 1045.05  462.77 1038.87  498.63 1035.18  520.21 1036.82   528.2 1039.99
  532.38 1042.63  546.02 1046.69  572.02 1058.67  599.08 1067.04  629.18 1071.19
  647.61  1072.1  656.76 1073.98  707.81 1079.37  780.82 1085.01  852.78 1088.55
#Mann= 3 , 0 , 0
       0     .11       0  450.54    .047       0  532.38     .11       0
Bank Sta=450.54,532.38
Exp/Cntr=0.3,0.1

Type RM Length L Ch R = 1 ,63065.05,311.62,311.62,239.08
XS GIS Cut Line= 5
  1343862.537075   795150.579314  1343574.796274   795087.667314
   1342978.95717   795522.638834  1342394.035825   795534.701938
  1342208.105201   795784.126323
#Sta/Elev= 30
       0 1089.89   51.66 1085.86  163.66 1073.39   239.3 1062.09  343.25 1056.37
  445.81 1058.36  499.76 1043.94  517.61 1043.34  534.79 1034.65  589.14 1035.65
  603.63 1034.64  606.48 1038.14  636.82 1045.18  708.02 1046.81  772.07  1052.4
  903.61 1058.72 1032.25 1068.11 1179.87 1066.89 1219.39 1065.09 1257.03 1065.87
  1282.9 1064.21    1360  1071.3 1444.72 1073.86 1613.47 1069.09 1646.32 1069.64
 1704.42 1065.96 1764.65 1064.94 1814.55  1066.6 1872.95 1064.02  1928.4 1067.43
#Mann= 3 , 0 , 0
       0     .12       0  517.61    .048       0  636.82     .12       0
#XS Ineff= 2 , 0
                          994.56         1074.73
Permanent Ineff=
       F       F
Bank Sta=517.61,636.82
Exp/Cntr=0.3,0.1

Type RM Length L Ch R = 1 ,62753.43,317.29,317.29,285.06
XS GIS Cut Line= 5
  1344043.049075   794987.012722  1343428.337266   794922.306162
   1342882.37605    795076.73317  1342202.324721   794930.312178
  1341909.005297    795303.43013
#Sta/Elev= 30
       0 1069.79   78.39 1070.04   178.3 1076.72  284.55 1070.14  440.88 1064.39
  459.25 1061.21  506.87 1058.34  622.75 1056.61  796.12 1046.45  812.15 1043.32
  831.88 1034.42  849.93 1035.88   906.3 1034.41  909.75 1040.07  933.21 1044.59
 1005.37 1042.29 1049.42 1046.21 1116.51 1063.28 1149.36 1068.17 1252.03  1068.8
 1320.02 1065.41 1351.99 1061.95  1542.8 1061.67 1610.74 1056.69 1765.94 1058.83
  1800.5 1057.55 1880.34 1063.12 2048.92 1062.81 2165.78 1067.57 2355.73 1080.28
#Mann= 3 , 0 , 0
       0     .11       0  812.15    .047       0  933.21     .11       0
Bank Sta=812.15,933.21
Exp/Cntr=0.3,0.1

Type RM Length L Ch R = 1 ,62436.14,590.68,590.68,551.64
XS GIS Cut Line= 3
  1343938.803315   794739.903986   1343463.10885   794656.570609
  1342155.249393    794805.31109
#Sta/Elev= 30
       0 1071.21   64.95 1067.46  166.81 1069.03  287.82 1066.51  399.65 1059.81
  467.61 1057.68  505.95 1058.03  529.99 1054.39  577.94 1051.38  723.75 1047.28
  763.26 1043.85   823.1 1045.19  842.28 1043.15  871.51 1036.52   892.9 1034.35
  919.35 1035.98  938.87 1039.69  944.26 1042.41  954.54 1044.37  996.13 1041.83
 1038.73 1043.18 1076.04 1048.24 1090.58 1052.36 1154.05 1059.59 1422.92 1073.94
 1463.52 1074.27 1506.62 1072.87  1562.9 1068.63  1640.8 1065.67 1799.23  1064.8
#Mann= 3 , 0 , 0
       0     .11       0   823.1    .047       0  954.54     .11       0
Bank Sta=823.1,954.54
Exp/Cntr=0.3,0.1

Type RM Length L Ch R = 1 ,61845.46,674.64,674.64,719.42
XS GIS Cut Line= 2
  1343699.342578   794171.412721  1342678.509298   794088.079345
#Sta/Elev= 30
       0 1067.63  104.62  1064.1  145.43 1064.35   172.2  1065.9  223.41 1065.11
  312.26 1059.34  359.09 1054.67  374.04 1054.69  455.11 1042.93  473.37 1041.81
  484.85 1042.73  487.39 1041.03  518.12 1035.24  541.77 1037.45  563.23 1034.23
  584.69 1037.48  587.76 1036.04  600.22 1038.95  602.66 1042.44  659.31 1041.62
  679.56  1042.9  722.53  1049.5  794.83 1066.39  875.14 1081.93  883.65 1082.33
  938.53 1090.42  959.79 1091.68  971.26 1093.56 1013.84  1094.7 1024.23  1093.9
#Mann= 3 , 0 , 0
       0     .11       0  484.85    .047       0  602.66     .11       0
#XS Ineff= 2 , 0
          400.87 1058.82
Permanent Ineff=
       F       F
Bank Sta=484.85,602.66
Exp/Cntr=0.3,0.1

Type RM Length L Ch R = 1 ,61170.81,415.38,415.38,401.56
XS GIS Cut Line= 5
  1344312.407539   794067.242225  1343302.134386   793427.824368
  1342951.350642   793478.237168  1342180.509681   793997.538545
  1340973.427952   793897.838577
#Sta/Elev= 30
       0 1059.52  102.85 1061.93  129.74 1065.05   241.8 1066.26  378.83 1057.05
  458.24 1056.54  531.75 1052.22  600.88 1054.63  647.65 1059.14  773.75 1058.21
 1100.33 1062.74 1197.06 1059.41 1294.86 1040.53 1349.09 1043.05 1362.35 1035.61
 1392.82 1032.87 1452.62 1040.34 1495.08 1042.74 1517.22 1047.46  1669.1 1052.81
 1916.12 1049.59 2053.08 1060.48 2262.77 1071.26 2362.81 1067.01 2479.45 1072.47
 2723.59 1058.17 2840.92 1059.51 3014.04 1044.32 3177.67 1048.25 3529.57 1048.73
#Mann= 3 , 0 , 0
       0     .11       0 1349.09    .047       0 1495.08     .11       0
#XS Ineff= 2 , 0
                         1745.38          1057.7
Permanent Ineff=
       F       F
Bank Sta=1349.09,1495.08
Exp/Cntr=0.3,0.1

Type RM Length L Ch R = 1 ,60755.43,566.02,566.02,413.41
XS GIS Cut Line= 3
  1343372.953714   793029.051504   1342817.39813   793070.718192
  1341918.489201   792574.897648
#Sta/Elev= 30
       0  1080.3  143.25  1064.9  267.22  1043.9  308.59 1040.55  330.93 1041.12
  340.95 1038.93  345.69  1033.9  367.36 1033.53  391.73 1030.33  409.14 1033.61
   434.4 1033.68  447.71 1038.75  483.97 1038.92   535.2 1050.57  575.78 1055.44
  644.77 1060.45  722.79 1059.58  805.05 1061.85   900.6 1067.42  976.98 1069.83
 1056.26 1070.92 1140.64 1067.76 1189.96 1069.64 1227.12 1066.66 1300.95 1069.15
 1309.28 1067.77 1382.81 1067.83 1439.36 1061.91  1461.4 1062.89  1583.7 1055.82
#Mann= 3 , 0 , 0
       0     .11       0  340.95    .047       0  447.71     .09       0
Bank Sta=340.95,447.71
Exp/Cntr=0.3,0.1

Type RM Length L Ch R = 1 ,60189.41,477.28,477.28,493.45
XS GIS Cut Line= 2
   1343554.94501   792854.549488  1342862.537074   792292.940399
#Sta/Elev= 30
       0 1077.78   47.52 1073.94  101.69 1067.36  131.69 1064.81  210.08 1052.53
  266.28 1040.37  313.26 1037.76  346.61 1040.74  363.06 1040.88  382.26 1037.69
  392.24 1037.83  399.02 1039.63  400.71 1038.21  407.15 1030.67  426.81 1032.74
  436.34  1031.4  451.58 1026.22  470.28 1032.76  497.15 1030.69  501.85 1037.98
  503.99  1041.1  541.91 1042.46  560.91 1044.92   598.4 1052.65  638.67 1059.31
  679.34  1062.1  703.17  1066.1  823.44 1078.06  837.35  1078.2  891.53 1083.01
#Mann= 3 , 0 , 0
       0     .09       0  400.71    .047       0  501.85      .1       0
Bank Sta=400.71,501.85
Exp/Cntr=0.3,0.1

Type RM Length L Ch R = 1 ,59712.13,490.45,490.45,511.24
XS GIS Cut Line= 2
  1344077.814771   792605.440368   1343227.12037   792022.107119
#Sta/Elev= 30
       0 1069.78  166.38 1065.84  285.52 1064.92  346.68 1062.56  408.07 1057.04
  427.16 1053.87  444.86 1053.31   517.5 1039.11  541.08 1038.26  554.24 1039.29
  561.15 1038.36  563.98 1035.19  572.16 1033.22  593.21 1035.05  599.27 1029.83
  613.75 1030.62   634.6 1022.11   656.8 1029.19  676.41 1028.03  677.69  1033.5
   679.7 1035.37  685.53 1039.24  693.34 1040.16  738.96 1039.99  764.42 1044.36
  782.33 1049.43  788.69 1049.28  806.71 1054.61  847.78 1060.61 1031.48 1080.18
#Mann= 3 , 0 , 0
       0      .1       0  593.21    .047       0   679.7      .1       0
Bank Sta=593.21,679.7
Exp/Cntr=0.3,0.1

Type RM Length L Ch R = 1 ,59221.69,400.33,400.33,350.99
XS GIS Cut Line= 2
  1344154.664819   792017.631215  1343555.055474   791691.459311
#Sta/Elev= 30
       0 1040.34   18.39 1040.26   38.26 1040.81   59.46 1039.99    83.9 1038.34
  116.17 1038.61  124.27 1038.23  151.91 1038.71  234.62 1037.19  266.46  1037.6
  272.39 1038.21  311.17 1037.95     343 1039.81  375.19  1040.8  378.56 1034.61
  385.42 1024.17  396.84 1024.84   419.7 1016.22  434.17 1024.56  444.07 1023.79
  447.64 1031.58  457.71  1036.1  471.72 1039.55  508.25 1038.46  519.39 1037.36
   541.6 1043.95  574.59 1052.97  612.29  1061.2  652.12 1066.65  682.58 1070.34
#Mann= 3 , 0 , 0
       0     .11       0  375.19    .047       0  457.71     .11       0
#XS Ineff= 2 , 0
          278.02 1050.94
Permanent Ineff=
       F       F
Bank Sta=375.19,457.71
Exp/Cntr=0.3,0.1

Type RM Length L Ch R = 1 ,58821.36,144.01,144.01,75.26
XS GIS Cut Line= 3
  1344212.638067   791772.502767  1344046.622451   791504.924655
  1343648.184946   791290.080878
#Sta/Elev= 30
       0 1060.09   34.46 1058.79   81.91 1055.78   138.8 1049.61  156.83 1046.97
  160.61 1045.81  224.17 1040.25  239.13 1039.72  267.66 1037.31  309.62 1037.24
  342.41 1038.37  358.56 1037.44  379.13    1038  381.29 1031.99  403.92 1022.97
  419.59 1021.24  434.39 1013.45  454.41 1021.24  461.37 1023.21  494.12 1023.27
  497.14 1026.69  522.42 1032.61  533.25  1036.5  571.06 1035.73  578.38 1036.39
  622.47 1036.16  642.23 1036.74  662.14 1038.32  738.05 1038.44  767.57  1039.9
#Mann= 3 , 0 , 0
       0     .11       0  379.13    .047       0  533.25     .11       0
#XS Ineff= 2 , 0
                          610.62         1049.97
Permanent Ineff=
       F       F
Bank Sta=379.13,533.25
Exp/Cntr=0.5,0.3

Type RM Length L Ch R = 1 ,58677.35,70.02,70.02,71
XS GIS Cut Line= 2
  1344227.567987   791688.895087  1343858.427379    791022.87947
#Sta/Elev= 30
       0 1058.91   52.52 1051.39  113.78 1045.31  131.66 1045.08  161.87 1042.19
  178.55 1039.44   184.1 1041.11  192.29 1039.74  201.73 1039.76   234.7 1041.27
  279.14 1036.84  290.55 1038.64  303.21 1038.35  309.96 1034.94  329.15  1023.5
  340.37 1020.34  357.78 1021.82  380.41 1013.61  408.27 1021.98  432.64 1021.16
  442.07 1035.44  444.01  1037.6  449.57 1037.25  453.15 1039.23   555.8 1043.69
  634.71 1051.14  645.38 1051.17  700.92  1055.5  734.05  1060.7  761.47 1061.74
#Mann= 3 , 0 , 0
       0     .11       0  309.96    .047       0  442.07     .11       0
Bank Sta=309.96,442.07
Exp/Cntr=0.5,0.3

Type RM Length L Ch R = 5 ,58642   ,,,
BEGIN DESCRIPTION:
Dam 37003-0095
END DESCRIPTION:
IW Pilot Flow=0
#Inline Weir SE= 30
       0 1059.95    8.41 1059.63   50.52 1052.96  110.03 1047.95  145.31 1045.57
  155.05 1045.78  178.27 1043.17  185.37 1043.76  193.13 1042.98  204.16 1044.51
  208.57 1044.18  229.59 1038.94  246.87 1026.41  271.75 1024.75  279.62 1025.11
  299.51 1024.09  301.79    1034  460.88    1034  466.49 1038.18  483.49 1038.56
  504.21 1040.41  535.41 1041.46  613.27 1048.34  667.21 1051.06  713.64 1056.46
  727.61 1056.93  734.26 1056.15  740.57 1056.76  746.19 1056.34  761.47 1060.64
IW Dist,WD,Coef,Skew,MaxSub,Min_El,Is_Ogee,SpillHt,DesHd
60,10,2.6,0,0.95,, 0 ,,,0,0,

Type RM Length L Ch R = 1 ,58607.33,197.65,197.65,191.93
XS GIS Cut Line= 2
  1344288.792947   791654.961007  1343919.652339    790988.94539
#Sta/Elev= 30
       0 1061.73   51.63 1055.87  108.08  1047.6  151.54 1042.88  172.08 1036.54
  190.82 1032.46  208.64 1030.71  223.56 1027.45  239.47 1027.83  277.69 1023.63
  309.23 1022.85  353.43 1022.07  369.97 1013.37  389.12 1021.08  398.89 1023.88
  427.43 1023.95  446.84 1032.15  474.02 1036.26  552.69 1039.36  604.82 1045.83
  624.46 1046.31  633.44 1045.44  653.96 1049.61  669.81 1051.52   686.4 1049.42
  702.18  1054.9   710.7 1055.75  721.81 1054.01  729.49 1056.76  761.47 1059.54
#Mann= 3 , 0 , 0
       0     .11       0  309.23    .047       0  398.89     .11       0
Bank Sta=309.23,398.89
Exp/Cntr=0.5,0.3

Type RM Length L Ch R = 1 ,58409.68,399.77,399.77,470.27
XS GIS Cut Line= 3
  1344717.467763   791825.187823  1344446.977395   791565.068527
  1344078.493043   790855.521774
#Sta/Elev= 30
       0 1078.34  166.97 1073.17  270.04 1066.92  311.03 1061.34  387.31 1053.97
  440.19 1043.76  492.92 1036.36  548.84 1022.18  562.25 1022.73  572.32    1021
  590.75 1020.49  620.74 1016.34  624.83 1014.08  635.91 1011.82   655.5 1012.78
  681.92 1016.28  697.42 1011.12  726.75 1016.62  741.79 1012.36  751.85 1011.04
  756.71 1013.76  757.14 1017.28  794.67 1017.99  822.01 1023.01  842.29 1029.27
  915.06 1042.54  956.05 1047.65 1013.24 1051.56 1091.56  1053.7 1174.79 1059.79
#Mann= 3 , 0 , 0
       0     .11       0  620.74    .047       0  757.14      .1       0
#XS Ineff= 2 , 0
          398.26  1060.3
Permanent Ineff=
       F       F
Bank Sta=620.74,757.14
Exp/Cntr=0.3,0.1

Type RM Length L Ch R = 1 ,58009.9 ,564.89,564.89,774.65
XS GIS Cut Line= 2
  1345273.539444   791683.642351  1344258.387315   790756.969198
#Sta/Elev= 30
       0 1040.55   51.44 1055.85   98.23  1065.9  158.63 1066.57  325.31 1053.92
  377.35 1047.75  422.17 1038.36  444.77 1036.53  467.79 1035.08  507.93 1036.05
  523.11 1040.13   549.2 1041.64  621.62 1037.07  696.86 1028.36  737.63 1018.99
  765.52 1016.53  783.19 1010.75  802.62 1006.89  860.72 1006.89  867.99 1012.02
  911.09 1014.29  953.71 1010.21  961.87 1013.58 1006.02  1013.5 1016.11 1018.24
 1041.75 1025.12 1138.51 1044.01 1175.14 1049.51 1285.89  1057.2  1374.5 1059.27
#Mann= 3 , 0 , 0
       0     .11       0  783.19    .047       0  867.99     .11       0
Bank Sta=783.19,867.99
Exp/Cntr=0.3,0.1

Type RM Length L Ch R = 1 ,57445.01,382.53,382.53,401.14
XS GIS Cut Line= 2
  1345207.399284   790442.860782  1344248.414835   790735.829614
#Sta/Elev= 30
       0 1079.95   47.52 1077.05   71.94 1078.86  102.49 1078.72  155.44 1074.88
  205.82 1073.28     245  1074.6  302.45 1071.43  335.76 1067.59  371.17 1061.54
   411.4 1051.07  469.05 1026.56  493.09  1017.4  501.05 1012.86  504.91 1010.82
  532.75 1003.17  554.95 1003.17  608.65 1013.75  626.66 1009.31  653.09 1014.31
  670.05  1014.2  688.95 1016.32  701.93 1018.59  728.46  1025.7  756.35 1027.33
  812.28 1038.48  882.89 1047.36  910.57 1052.05  938.28 1055.04 1002.74 1059.51
#Mann= 3 , 0 , 0
       0     .11       0  501.05    .047       0  608.65     .11       0
Bank Sta=501.05,608.65
Exp/Cntr=0.3,0.1

Type RM Length L Ch R = 1 ,57062.48,660,660,342.32
XS GIS Cut Line= 3
  1345146.418292   790298.013165  1344723.504499   790175.052269
  1344164.430451   790404.349933
#Sta/Elev= 30
       0 1070.25   35.33 1066.82   57.07 1066.82   99.41 1062.45  112.76 1062.71
  198.52 1056.66  413.43 1035.32  452.55 1033.12  527.56 1020.96  550.46 1013.79
  583.34 1011.66  586.84 1009.41   603.5 1006.87  628.07  1009.3  645.05 1001.97
  660.72 1009.08   681.9 1008.48  686.73 1007.12  703.81 1008.75  709.91 1012.45
   751.6 1011.33  808.86 1012.74  816.09 1016.16  836.77 1019.09  845.43 1022.75
  859.21 1030.36  899.28 1040.45  960.88 1051.28  985.28 1053.42  1044.7 1061.43
#Mann= 3 , 0 , 0
       0     .11       0  583.34    .047       0  709.91     .11       0
Bank Sta=583.34,709.91
Exp/Cntr=0.3,0.1

Type RM Length L Ch R = 1 ,56402.48,551.29,551.29,848.93
XS GIS Cut Line= 5
  1346138.652021   790213.478893  1345059.612788   790013.290861
  1344930.797044   790087.660653  1344708.918259   789607.040877
  1344056.140531   789548.013165
#Sta/Elev= 30
       0 1051.01  279.95 1041.03  344.76 1036.13  442.51 1034.65  472.11 1037.11
  580.97 1031.38  622.34 1032.94  663.26 1038.07  711.58 1037.72  760.88 1033.39
  894.58 1031.98 1040.49 1032.74 1246.19 1038.34  1405.3 1011.92 1497.44 1011.24
  1523.4 1005.94 1539.72 1006.27 1558.76  997.73 1580.52 1005.44 1609.48 1005.46
 1613.17 1010.94 1619.74 1021.69 1663.64 1043.71 1738.24  1055.9 1842.03 1068.62
 1912.87 1073.56 2187.78 1068.86 2263.46 1070.49 2375.31 1087.66    2431 1093.61
#Mann= 3 , 0 , 0
       0     .11       0 1497.44    .047       0 1613.17     .11       0
#XS Ineff= 2 , 0
         1003.81 1050.89
Permanent Ineff=
       F       F
Bank Sta=1497.44,1613.17
Exp/Cntr=0.3,0.1

Type RM Length L Ch R = 1 ,55851.19,393.11,393.11,437.47
XS GIS Cut Line= 3
  1345662.887156   789272.472044  1344830.446068   789544.540909
  1344469.335027   789447.318637
#Sta/Elev= 30
       0 1130.09   67.42 1126.16  187.36 1113.22   249.8 1103.22  285.68  1095.9
  302.66 1090.63  314.57 1088.93  350.56  1074.3  370.48 1070.29  398.06  1059.5
  417.64 1045.98  453.52 1028.65  474.17 1023.84  487.83 1011.21  491.91 1007.23
     497 1005.61  525.57 1006.48  539.28   995.1  552.99 1004.51   562.3 1008.66
  573.75 1006.51  582.61 1007.53  590.95 1010.78  632.72 1009.09  735.16 1014.86
  749.63 1016.76  798.51 1028.39 1011.08 1058.08 1175.24 1063.74 1249.74 1070.62
#Mann= 3 , 0 , 0
       0     .11       0  487.83    .047       0  590.95     .11       0
Bank Sta=487.83,590.95
Exp/Cntr=0.3,0.1

Type RM Length L Ch R = 1 ,55458.08,280.87,280.87,292.39
XS GIS Cut Line= 2
  1345291.220852   788906.031852  1344509.970931   789371.309549
#Sta/Elev= 30
       0  1083.6    54.1 1083.57  113.37 1080.29  133.06 1078.45   167.6 1072.65
   185.9 1068.67  206.98 1061.91  221.87 1058.82  243.99  1047.9  272.45 1044.58
  281.66 1041.15  296.16 1030.43  300.73 1028.81  322.72 1011.11  338.41 1003.15
  347.12 1005.94   366.7  990.01   385.2 1004.46  399.35    1002  433.57 1010.17
  447.98 1007.69  454.99 1007.73  475.42  1009.3  522.34 1010.75  556.51 1012.82
   568.2 1014.41  607.09 1022.97  807.51 1045.92  828.58 1049.49   909.3 1060.27
#Mann= 3 , 0 , 0
       0      .1       0  322.72    .047       0  433.57      .1       0
Bank Sta=322.72,433.57
Exp/Cntr=0.3,0.1

Type RM Length L Ch R = 1 ,55177.21,242.42,242.42,210.41
XS GIS Cut Line= 3
  1345210.926324   788761.702764  1345010.112628   788731.488492
  1344456.178547     789106.0915
#Sta/Elev= 30
       0 1048.31   27.69 1046.13   38.61  1047.2   50.67 1045.33   94.53 1042.34
  131.86 1041.12  203.01 1034.35  217.38 1034.28  259.07 1031.36  291.68 1025.56
   310.3 1023.98     338 1014.74  373.17 1009.71  380.89 1007.04  391.19 1005.78
  401.52  999.82  415.67 1001.92  439.61     988  455.93 1000.81  462.46  998.71
     494 1005.21  497.38    1008  502.26  1009.5  514.58 1008.34  569.74 1007.67
  641.29 1013.77  697.86 1030.62  757.57 1043.92  806.55 1052.44  871.78 1061.65
#Mann= 3 , 0 , 0
       0      .1       0  380.89    .047       0  497.38      .1       0
#XS Ineff= 2 , 0
          280.74 1034.57
Permanent Ineff=
       F       F
Bank Sta=380.89,497.38
Exp/Cntr=0.5,0.3

Type RM Length L Ch R = 1 ,54934.79,97.3,97.3,94.85
BEGIN DESCRIPTION:
Upstream xs of Bridge 37003-0046
END DESCRIPTION:
XS GIS Cut Line= 6
  1345007.963252   788301.162988  1344868.776436   788574.778092
  1344576.998387   788706.449132  1344450.499571   788692.208748
  1344310.535923   788532.416236  1344115.782131   788618.107884
#Sta/Elev= 30
       0  1057.8  22.981  1052.9  48.225  1049.6  86.196  1041.9 119.855  1037.1
 144.038  1034.8 164.756  1028.7  176.07  1026.5 252.649  1018.3 286.449  1016.5
 302.359  1013.9  316.43  1009.7  341.68   993.9  349.29  996.85  363.44  986.68
  384.11  996.63  391.73  994.23 409.768  1006.6 409.768  1006.7 445.194  1009.9
 497.379  1020.6  531.32  1020.1  575.09  1025.4 590.505  1025.6 609.526  1024.3
 640.214  1019.3 691.126  1018.4 722.027  1022.3 751.372  1024.2 841.598  1042.9
#Mann= 3 , 0 , 0
       0      .1       0  316.43    .047       0 409.768      .1       0
#XS Ineff= 2 , 0
       0 283.126  1019.4 465.701       0  1019.4
Permanent Ineff=
       F       F
#Block Obstruct= 2 , 0
          213.28 1034.47
Bank Sta=316.43,409.768
Skew Angle= 45
Exp/Cntr=0.5,0.3

Type RM Length L Ch R = 3 ,54889.68,,,
BEGIN DESCRIPTION:
Bridge : 37003-0046 - SR-1110 / Liledoun Rd
END DESCRIPTION:
Bridge Culvert--1,0,-1,-1, 0
Deck Dist Width WeirC Skew NumUp NumDn MinLoCord MaxHiCord MaxSubmerge Is_Ogee
29.1,32,2.6,45, 154, 154, , , 0.95, 0, 0,0,,
  16.193  17.678  19.375  25.314   29.84  31.113  40.164  50.558  57.912  60.882
  71.206  71.559  83.863   89.52  96.167 107.622  108.47 110.309 119.925 123.178
 131.451 138.593 142.977 153.937 154.503 163.695 168.928  173.17 181.302 182.504
 183.282 190.919 196.646 199.333 203.859 219.415  222.88 227.193 230.375 239.426
 243.033 253.215 255.195 263.256  264.67 272.519 278.247 280.014 283.691 287.015
 288.712 296.348  301.44 303.702 303.702 445.124 445.124 446.962 452.619 455.023
 461.529 467.256 470.014  471.64 473.832 477.792 479.348  485.57 489.601 491.439
 492.712 499.288 501.268 505.652 511.733 512.511 516.612 519.794 526.653 527.784
  531.32 533.512 535.492 541.644 545.321 548.573 552.321 554.301 556.705 560.029
 563.211 566.039 571.767 574.383  578.06  581.03 586.121 593.616 601.819 602.384
 609.031 617.941 623.385 623.951 624.941 632.436 639.295 639.719 648.134 650.114
 655.276 656.619 663.832 665.317 670.125 672.246  681.58 682.287 685.328 690.631
 691.904 698.268 705.268 705.622 706.188 712.269 720.118 727.896 729.168 729.805
 731.926 739.139 746.846 750.665 752.291 760.988  762.19 772.938 775.625 782.414
 786.586 790.545 795.212 800.091 805.112 809.567 812.961 819.112 821.658 823.072
 829.153 832.972 838.416 842.164
  1050.2  1050.1  1049.8    1049  1048.3  1048.1  1046.9  1045.2  1044.1  1043.7
  1042.5  1042.4  1040.4  1039.6  1038.6  1036.9  1036.8  1036.5  1035.2  1034.7
  1033.6  1032.7  1031.9  1030.5  1030.5    1029  1028.2  1027.6  1026.7  1026.5
  1026.5  1025.6  1025.1  1024.8  1024.5  1023.1  1022.9  1022.5  1022.3  1021.7
  1021.5  1021.1    1021  1020.5  1020.5  1020.3  1020.2  1020.2    1020  1019.8
  1019.8  1019.7  1019.8    1020    1020    1020    1020    1020  1019.7  1019.8
  1019.8  1019.9  1019.8  1019.9  1019.7  1019.6  1019.6  1019.5  1019.4  1019.2
  1019.3  1019.6  1019.6  1019.5  1019.5  1019.6  1019.5  1019.5  1019.7  1019.7
  1019.6  1019.5  1019.5  1019.7  1019.6  1019.6  1019.5  1019.5  1019.5  1019.3
  1019.3  1019.2  1019.1    1019  1018.9  1018.7  1018.5  1018.2  1018.1  1018.1
  1017.6  1017.3  1016.9  1016.9  1016.8  1016.5  1016.3  1016.3  1015.7  1015.6
  1015.2  1015.2  1014.8  1014.7  1014.5  1014.4  1014.8  1014.8  1015.6  1017.2
  1017.6  1019.5  1021.3  1021.4  1021.5  1022.7  1023.6  1024.1  1024.1  1024.2
  1024.2  1024.5  1024.9  1025.2  1025.2  1025.3  1025.5  1025.8  1026.6  1028.9
  1030.4  1031.9  1033.5  1034.7    1035  1035.6  1036.1  1037.4  1037.7  1037.9
  1038.5    1039  1039.6  1039.8
                                                                                
                                                                                
                                                                                
                                                                                
                                                                                
                                  1017.5  1017.5
                                                                                
                                                                                
                                                                                
                                                                                
                                                                                
                                                                                
                                                                                
                                                                                
                                                                                
                                
  -5.515  -4.031  -2.333   3.606   8.132   9.405  18.455   28.85  36.204  39.174
  49.497  49.851  62.155  67.812  74.458  85.913  86.762    88.6  98.217  101.47
 109.743 116.885 121.269 132.229 132.795 141.987  147.22 151.462 159.594 160.796
 161.574 169.211 174.938 177.625 182.151 197.707 201.172 205.485 208.667 217.718
 221.324 231.507 233.487 241.548 242.962 250.811 256.538 258.306 261.983 265.306
 267.004  274.64 279.731 281.994 281.994 423.416 423.416 425.254 430.911 433.315
  439.82 445.548 448.306 449.932 452.124 456.084 457.639 463.862 467.893 469.731
 471.004  477.58  479.56 483.944 490.025 490.803 494.904 498.086 504.945 506.076
 509.612 511.804 513.784 519.936 523.613 526.865 530.613 532.593 534.997  538.32
 541.502 544.331 550.058 552.675 556.352 559.321 564.413 571.908  580.11 580.676
 587.323 596.232 601.677 602.243 603.233 610.728 617.587 618.011 626.426 628.406
 633.568 634.911 642.124 643.609 648.417 650.538 659.872 660.579  663.62 668.923
 670.196  676.56  683.56 683.914 684.479  690.56 698.409 706.188  707.46 708.097
 710.218  717.43 725.138 728.956 730.583  739.28 740.482  751.23 753.917 760.706
 764.877 768.837 773.504 778.383 783.404 787.858 791.253 797.404  799.95 801.364
 807.445 811.264 816.708 820.456
  1050.2  1050.1  1049.8    1049  1048.3  1048.1  1046.9  1045.2  1044.1  1043.7
  1042.5  1042.4  1040.4  1039.6  1038.6  1036.9  1036.8  1036.5  1035.2  1034.7
  1033.6  1032.7  1031.9  1030.5  1030.5    1029  1028.2  1027.6  1026.7  1026.5
  1026.5  1025.6  1025.1  1024.8  1024.5  1023.1  1022.9  1022.5  1022.3  1021.7
  1021.5  1021.1    1021  1020.5  1020.5  1020.3  1020.2  1020.2    1020  1019.8
  1019.8  1019.7  1019.8  1019.9  1019.9  1019.9  1019.9    1020  1019.7  1019.8
  1019.8  1019.9  1019.8  1019.9  1019.7  1019.6  1019.6  1019.5  1019.4  1019.2
  1019.3  1019.6  1019.6  1019.5  1019.5  1019.6  1019.5  1019.5  1019.7  1019.7
  1019.6  1019.5  1019.5  1019.7  1019.6  1019.6  1019.5  1019.5  1019.5  1019.3
  1019.3  1019.2  1019.1    1019  1018.9  1018.7  1018.5  1018.2  1018.1  1018.1
  1017.6  1017.3  1016.9  1016.9  1016.8  1016.5  1016.3  1016.3  1015.7  1015.6
  1015.2  1015.2  1014.8  1014.7  1014.5  1014.4  1014.8  1014.8  1015.6  1017.2
  1017.6  1019.5  1021.3  1021.4  1021.5  1022.7  1023.6  1024.1  1024.1  1024.2
  1024.2  1024.5  1024.9  1025.2  1025.2  1025.3  1025.5  1025.8  1026.6  1028.9
  1030.4  1031.9  1033.5  1034.7    1035  1035.6  1036.1  1037.4  1037.7  1037.9
  1038.5    1039  1039.6  1039.8
                                                                                
                                                                                
                                                                                
                                                                                
                                                                                
                                  1017.4  1017.4
                                                                                
                                                                                
                                                                                
                                                                                
                                                                                
                                                                                
                                                                                
                                                                                
                                                                                
                                
Pier Skew, UpSta & Num, DnSta & Num=  ,339.058, 2 ,317.35, 2 , 0 , 0 , 0 ,,
       1       1
  1002.7    1018
       1       1
 1002.61 1017.91
Pier Skew, UpSta & Num, DnSta & Num=  ,374.413, 2 ,352.705, 2 , 0 , 0 , 0 ,,
       1       1
  1006.1    1018
       1       1
 1006.01 1017.91
Pier Skew, UpSta & Num, DnSta & Num=  ,409.768, 2 ,388.06, 2 , 0 , 0 , 0 ,,
       1       1
  1005.7    1018
       1       1
 1005.61 1017.91
BR Coef=-1 , 1 , 0 ,, 0 ,,,0.8,0,1.2,0,
WSPro=,,,, 1 ,,,, 0 ,,,, 0 ,,,,-1 ,-1 ,-1 , 0 , 0 , 0 , 0 , 0
BC Design=,, 0 ,, 0 ,,,,,,

Type RM Length L Ch R = 1 ,54837.49,468.52,468.52,470.76
BEGIN DESCRIPTION:
Down stream xs of Bridge 37003-0046
END DESCRIPTION:
XS GIS Cut Line= 6
  1344940.038388   788252.816747  1344824.342388    788491.89694
  1344556.550003   788612.178924  1344483.830131   788602.981996
  1344330.825075   788420.001004  1344086.125683   788527.668716
#Sta/Elev= 30
       0  1055.9   4.667  1055.1  15.839  1048.4  27.365  1045.7 106.915  1039.2
 119.572  1034.1 144.957  1031.6 173.312  1024.4 231.931  1021.2 245.366  1015.8
 273.721  1010.2 294.722  1009.6  315.56 1001.56  340.59  985.91  388.06  1006.6
 412.809  1009.4 428.153  1009.1 469.519  1013.6 508.763  1015.1 534.502  1012.5
 576.575    1012 592.273  1009.4 636.184  1009.2 650.043    1013 671.186  1013.8
 690.278  1022.4 710.996  1025.3 752.079  1024.9 793.869  1034.3 810.486  1036.1
#Mann= 3 , 0 , 0
       0      .1       0 294.722    .047       0 412.809      .1       0
#XS Ineff= 2 , 0
       0 256.397    1014     493       0    1014
Permanent Ineff=
       F       F
#Block Obstruct= 2 , 0
          221.98 1030.62
Bank Sta=294.722,412.809
Skew Angle= 45
Exp/Cntr=0.5,0.3

Type RM Length L Ch R = 1 ,54368.96,156.25,156.25,58.78
XS GIS Cut Line= 2
  1344910.280052   787950.329707  1343920.045683   788410.290668
#Sta/Elev= 30
       0  1049.1   54.57 1049.32  100.95 1045.13  200.37 1043.58  260.25 1037.13
  282.84  1027.9   339.7 1028.24  363.95  1019.2  397.02 1020.59  457.75 1017.66
  501.62 1006.18  542.21 1007.95  550.75 1006.92  553.65  1002.5  584.98 1006.43
  599.35 1004.99  605.88 1001.35  613.71  983.06  628.07  989.77  646.35 1003.08
   655.5 1005.38  677.69 1005.07     692 1008.67  748.06 1006.96  861.86    1018
  922.94 1018.95  940.02 1022.06  958.71 1029.65   977.5    1032 1091.85 1033.97
#Mann= 3 , 0 , 0
       0      .1       0  599.35    .047       0   655.5      .1       0
#XS Ineff= 2 , 0
          532.47 1011.81  696.31         1011.91
Permanent Ineff=
       F       F
#Block Obstruct= 2 , 0
          440.04  1028.5
Bank Sta=599.35,655.5
Exp/Cntr=0.5,0.3

Type RM Length L Ch R = 1 ,54212.71,79.24001,79.24001,22.46
XS GIS Cut Line= 5
  1344549.479027   788060.825195  1344417.645043   788101.168107
  1344384.048627   788031.146731  1344015.562099   788171.452267
  1343970.393587   788261.789035
#Sta/Elev= 30
       0 1017.47   24.29 1018.22   34.88 1016.22   60.64 1016.66   82.09 1014.95
  121.65  1007.4   200.7 1008.49  237.15 1006.59   248.1  987.31  251.81  983.83
  296.58  985.36  315.13  980.66  340.37  985.66  345.59  984.02  375.69  983.84
   376.2  983.93  377.12   988.2   380.4 1005.06  380.79 1005.39  439.26 1008.83
  448.42 1013.26  460.64 1013.17  475.12 1017.31  497.17 1020.09  535.25 1022.08
  609.83 1036.59  640.57 1038.85  663.81 1037.97  674.26  1035.2  710.83 1038.79
#Mann= 3 , 0 , 0
       0      .1       0   248.1    .047       0  377.12      .1       0
#Block Obstruct= 2 , 0
          116.65 1023.58
Bank Sta=248.1,377.12
Exp/Cntr=0.5,0.3

Type RM Length L Ch R = 5 ,54177   ,,,
BEGIN DESCRIPTION:
DAM
END DESCRIPTION:
IW Pilot Flow=0
#Inline Weir SE= 30
       0 1016.98   25.68 1017.84    37.9 1014.59   64.37 1014.78   85.89 1012.56
  112.43  1008.3  122.35 1007.71  167.43 1006.68   201.2 1007.55  210.12 1008.57
  220.62  995.23   225.9  996.74  234.02     995  399.04     995   406.4  992.43
  411.66  992.07  419.91  993.67  427.88  993.52  434.45  995.46  462.22  998.97
  495.88 1013.17   516.9 1018.68   533.6 1021.48  562.49 1023.59  660.58 1040.67
  690.27 1043.96  737.57 1046.34  749.13 1046.11  766.17 1041.06  775.22 1041.22
IW Dist,WD,Coef,Skew,MaxSub,Min_El,Is_Ogee,SpillHt,DesHd
69,10,2.6,0,0.95,, 0 ,,,0,0,

Type RM Length L Ch R = 1 ,54133.48,311.23,311.23,440.38
XS GIS Cut Line= 5
  1344545.640307   788039.711851  1344438.154099   788070.422251
  1344396.034035   787951.668587  1343965.154291   788116.382699
  1343907.783667   788231.123947
#Sta/Elev= 30
       0 1016.77   24.76 1017.63   38.08 1013.53   61.07 1013.35  111.79 1008.16
  144.03 1006.79  189.77 1008.31  200.56  994.68   219.9  983.69  235.78  988.81
  237.79   988.5   272.2   980.2  286.23  982.85  327.43     985  352.52  983.53
  378.11  985.11  439.72  983.82  461.33  997.19  472.37 1001.62  479.73 1008.79
  505.21 1014.79  520.21 1015.34  559.81 1023.67  583.67  1024.5  661.43 1037.28
  678.68 1041.47  710.98 1045.66  754.54 1046.37  787.98 1049.08  827.36 1047.08
#Mann= 3 , 0 , 0
       0     .11       0  237.79    .047       0  327.43     .09       0
#Block Obstruct= 2 , 0
          110.99 1022.13
Bank Sta=237.79,327.43
Exp/Cntr=0.5,0.3

Type RM Length L Ch R = 1 ,53822.24,525.64,525.64,334.03
XS GIS Cut Line= 6
  1344672.700787   787901.257451  1344573.091315   787830.945003
  1344560.823283   787662.671083  1344130.159219   787708.813675
  1344092.668403   787769.101035  1343882.829555   787840.512235
#Sta/Elev= 30
       0 1020.51   74.76 1012.35  189.77 1002.12  290.45  998.03  351.59  994.01
   437.6  991.95  474.19  992.47  495.89   982.7  510.88  978.33  516.94  979.16
  539.11  978.17  561.17  979.16   586.6  978.48  601.75  983.61  616.07  985.86
  655.25  988.53  667.38  991.46   677.1   995.6  702.12  997.75  723.82  1009.7
  794.81 1024.65  800.21 1026.93   822.3 1031.31  833.86 1035.28  847.82  1037.7
  880.24  1038.7  894.41 1043.59  940.44 1051.55  955.37 1055.49 1016.47 1063.34
#Mann= 3 , 0 , 0
       0     .11       0  495.89    .047       0  601.75     .09       0
#XS Ineff= 2 , 0
                          712.95          1020.9
Permanent Ineff=
       F       F
#Block Obstruct= 2 , 0
          335.58 1015.49
Bank Sta=495.89,601.75
Exp/Cntr=0.3,0.1

Type RM Length L Ch R = 1 ,53296.6 ,317.13,317.13,181.94
XS GIS Cut Line= 5
  1344921.166964   787744.519147  1344786.401267   787631.726187
  1344569.715571   787611.892203  1344626.333811   787332.845291
  1344106.659571   787088.173802
#Sta/Elev= 30
       0 1020.09    22.8 1008.19   63.22 1008.29   271.9  997.22  436.88  997.08
  470.11  983.81  491.04  977.57  519.54  976.82  549.34   977.2  554.22  979.79
  567.91  981.05  570.85  983.81  586.11  995.62  596.32   998.1  612.59 1005.85
  647.72 1029.81  663.97  1037.1  678.06 1040.47  715.07 1041.76  809.38 1028.66
  875.83 1018.91  918.21  1005.6  929.53 1005.74   989.1 1022.41 1043.94 1027.24
 1046.01 1025.47 1056.21 1025.33 1099.98 1028.35 1229.69 1026.84 1252.45 1029.49
#Mann= 3 , 0 , 0
       0     .11       0  470.11    .047       0  570.85     .11       0
Bank Sta=470.11,570.85
Exp/Cntr=0.3,0.1

Type RM Length L Ch R = 1 ,52979.47,286.88,286.88,248.67
XS GIS Cut Line= 3
  1345510.432628   787888.142955    1344921.1749   787605.542123
  1344850.862324   787185.864426
#Sta/Elev= 30
       0 1020.37   55.04 1013.56  128.92 1012.92  222.03  1009.6  262.73 1003.43
   278.6  999.43  305.82  997.74  337.07  999.41  508.67  995.25  582.61 1000.87
  614.21  998.91  631.48 1002.38  653.52  999.89  661.01  995.92  702.42  986.02
  705.17  983.43  707.93  980.85  729.24  977.67  751.18  976.67  790.95  977.86
  799.26  983.05  807.51  986.92   840.2  990.96  860.68  996.72  883.52  995.51
  896.27  997.07  915.29 1002.39  957.97 1025.87 1032.27 1042.94 1079.05 1050.16
#Mann= 3 , 0 , 0
       0      .1       0  705.17    .047       0  799.26      .1       0
#XS Ineff= 2 , 0
           612.4 1010.01
Permanent Ineff=
       F       F
Bank Sta=705.17,799.26
Exp/Cntr=0.3,0.1

Type RM Length L Ch R = 1 ,52692.6 ,378.35,378.35,453.33
XS GIS Cut Line= 3
  1345504.670964   787726.635883  1345240.999028   787562.573419
   1345008.57714   787058.667114
#Sta/Elev= 30
       0 1029.93   99.79 1027.57  113.43 1026.74  145.81 1022.04   168.7 1026.26
  186.95 1022.04  195.76 1022.67  215.13 1018.43  244.45 1019.86  271.09 1018.12
  295.15 1014.17  311.54  1009.5  328.94 1001.53   338.1   996.4  353.77  985.63
  356.06  984.92  367.45  983.78  399.41  986.16  406.21  983.57  414.91  976.44
  451.42  974.71  483.81  975.22  499.08  982.51  520.36  992.97  569.38     996
  636.84 1003.54  661.68 1005.05  763.15  1015.6  826.18 1019.14  865.47  1018.9
#Mann= 3 , 0 , 0
       0     .11       0  406.21    .047       0  499.08     .11       0
Bank Sta=406.21,499.08
Exp/Cntr=0.3,0.1

Type RM Length L Ch R = 1 ,52314.24,437.12,437.12,446.34
XS GIS Cut Line= 2
  1345914.827253   787480.542187  1345086.702196   786957.104618
#Sta/Elev= 30
       0  998.34   14.68  997.21   40.96  999.79   81.68  996.58  136.87 1001.53
  204.23  999.98  290.55 1003.18  353.51 1001.98  416.93 1004.23  452.75 1000.98
  470.07  997.48  497.09  988.22  504.83  987.95  511.07  984.92  523.35  978.13
  557.15  973.67  579.32   976.5  591.39  976.47  602.59  985.93  625.35  990.81
  655.84  993.78  699.26  994.96  813.38   994.5  863.54  998.23  878.26 1001.34
  890.76 1000.11  911.21 1001.25   930.9 1008.11  947.31 1005.22  979.68 1007.59
#Mann= 3 , 0 , 0
       0     .11       0  511.07    .047       0  602.59     .11       0
#XS Ineff= 2 , 0
           422.2 1007.26
Permanent Ineff=
       F       F
Bank Sta=511.07,602.59
Exp/Cntr=0.3,0.1

Type RM Length L Ch R = 1 ,51877.12,478.64,478.64,481.65
XS GIS Cut Line= 2
  1345936.311541   786961.010922   1345291.78034   786593.823338
#Sta/Elev= 30
       0 1040.99   27.39 1037.98   42.37 1033.01   98.11 1021.54  119.61 1017.56
  161.51 1011.91  215.31  999.63  262.67  986.93  275.63  986.38  288.63  979.95
  293.26  976.54  296.23  975.47  306.32  974.04  318.47   974.5  340.92     973
  363.36  974.52   377.3  980.31  390.43  994.68  418.06  992.32  438.96  992.37
  470.22  990.64   513.7  992.24  537.59  994.58  546.65  996.69  557.27  999.95
  575.99 1007.96   655.1 1046.78  686.12 1057.14  719.09 1066.68  741.79 1070.64
#Mann= 3 , 0 , 0
       0     .11       0  288.63    .047       0   377.3     .11       0
Bank Sta=288.63,377.3
Exp/Cntr=0.3,0.1

Type RM Length L Ch R = 1 ,51398.48,573.14,573.14,524.93
XS GIS Cut Line= 2
  1346168.733429   786537.182826  1345543.733492    786193.43281
#Sta/Elev= 30
       0 1029.69   45.59 1023.59   67.01 1022.01   94.19 1013.59  120.96 1007.89
  182.89  996.53  212.84  992.76   246.8  990.64  262.34  988.94   287.2  988.67
  296.28  986.54  302.58  982.65  315.71   974.2   336.9  977.51  352.17   973.8
  359.34  972.98  381.77  977.52  388.43  975.49  398.68  983.47  422.08  990.62
  480.03  987.75  497.93  988.62  517.19  994.63  558.85 1018.29  572.61 1025.29
  589.73 1031.99  608.74 1038.34  627.67 1040.83  654.75 1042.71  713.29 1049.27
#Mann= 3 , 0 , 0
       0     .11       0  302.58    .047       0  398.68     .11       0
Bank Sta=302.58,398.68
Exp/Cntr=0.3,0.1

Type RM Length L Ch R = 1 ,50825.34,682.61,682.61,654.33
XS GIS Cut Line= 2
  1346492.952181   786205.151466  1345818.473076   785587.964009
#Sta/Elev= 30
       0 1020.71   228.9  995.23   243.4  992.22  264.31     990  286.17  988.36
  331.56  989.38  352.87   988.1  371.97  989.11  437.18  988.48  452.14  987.24
  478.56  978.18  483.77  975.87  512.18  974.57  527.58     972  550.45   976.2
  570.74  973.81  573.56  974.89  580.06  981.47  596.08   986.6   606.4  992.92
  634.05 1013.05  652.62 1022.76  682.58 1031.07  698.53 1033.49  731.92 1034.54
  753.03 1036.52  762.64 1038.95   793.1 1042.33  821.36 1047.28  914.24 1048.26
#Mann= 3 , 0 , 0
       0     .11       0  478.56    .047       0  580.06      .1       0
Bank Sta=478.56,580.06
Exp/Cntr=0.3,0.1

Type RM Length L Ch R = 1 ,50142.73,259.76,259.76,245.28
XS GIS Cut Line= 3
  1346938.264693   785978.589033  1346753.368821   785582.755689
  1346391.389685   785142.651497
#Sta/Elev= 30
       0 1009.94   46.29 1007.33   67.01 1004.64  166.29 1001.72  191.52  1000.1
  215.12  996.99  272.27  996.76   302.3  999.11  340.74   999.9  471.67   997.4
  498.58  995.31   540.4   984.9  563.51  984.65  573.23  979.97  581.46  975.82
  617.34  974.87  639.78  971.26  662.21  974.85  688.52  973.44  697.28  980.38
  699.79  983.16  705.39  982.17  758.56  992.92  786.78 1003.75  807.16 1013.62
  832.72 1022.57  871.45 1033.95  926.64 1043.96  940.01 1047.87 1006.73 1049.66
#Mann= 3 , 0 , 0
       0     .11       0  573.23    .047       0  697.28     .11       0
#XS Ineff= 2 , 0
          416.54  1006.1
Permanent Ineff=
       F       F
Bank Sta=573.23,697.28
Exp/Cntr=0.3,0.1

Type RM Length L Ch R = 1 ,49882.96,489.78,489.78,507.89
XS GIS Cut Line= 3
  1347151.806326   785788.484841   1347045.03551   785572.339049
  1346615.348085   784965.568232
#Sta/Elev= 30
       0 1019.29  152.75 1017.35  251.38  1014.2  316.16 1010.53  451.25  997.57
  487.87  992.21  534.97  983.17  545.32  983.95  560.15  981.88  566.93  982.77
  577.47  980.98  587.86  974.85  603.94  976.58  612.86  975.34  626.51  970.88
  649.09  976.77  661.63  975.43  684.04  975.58  686.55  980.51  702.59  986.33
  709.54  986.59  733.89  994.86  752.41 1003.31   758.2 1008.64   774.5 1014.05
  799.17 1024.84  813.74 1027.86   850.7 1038.58  872.21 1041.94  984.59 1045.97
#Mann= 3 , 0 , 0
       0     .11       0  577.47    .047       0  686.55     .15       0
Bank Sta=577.47,686.55
Exp/Cntr=0.3,0.1

Type RM Length L Ch R = 1 ,49393.18,608.28,608.28,806.58
XS GIS Cut Line= 2
  1347433.056374   785223.380713  1346961.702262   784671.297384
#Sta/Elev= 30
       0 1041.03   58.96 1030.86  107.31  1017.8   118.7  1015.3  160.35 1000.23
  182.61  993.71   204.2  985.26  219.97  983.03  239.03  981.58  274.39  980.12
  282.01  978.07  292.33  972.35  314.26  973.33  328.02  971.31  336.81  970.97
  346.72  971.48  359.36  973.34  377.38  972.33  386.51  977.77  393.97  982.55
  429.24  992.59  433.12  994.95  460.88 1000.39  478.68 1005.86   508.9 1010.34
  574.59 1021.64  618.35 1026.81  659.28 1029.29  700.44 1030.45  725.93 1030.32
#Mann= 3 , 0 , 0
       0     .11       0  282.01    .047       0  386.51     .11       0
Bank Sta=282.01,386.51
Exp/Cntr=0.3,0.1

Type RM Length L Ch R = 1 ,48784.89,587.18,587.18,480.33
XS GIS Cut Line= 2
   1347779.41055   784387.443176  1347011.181302   784478.589032
#Sta/Elev= 30
       0 1049.28   23.77 1050.57  125.99 1049.22  163.37 1043.39  188.36 1038.08
   211.4  1031.9  228.18 1029.83  239.82 1027.62  271.01 1015.09  279.76 1005.63
  294.12   993.5  304.58  981.63  307.29  979.15  313.42  970.66  335.01  971.71
  357.53  969.23  380.06  971.71  384.24  971.06  391.28  975.74  393.36  979.48
  396.54  982.98   409.8  982.65  445.86  983.66  483.82  987.03  527.23  992.81
  569.76    1001  610.27 1007.73  692.31 1017.44  739.87 1019.83  773.62 1020.14
#Mann= 3 , 0 , 0
       0      .1       0  307.29    .047       0  396.54     .11       0
Bank Sta=307.29,396.54
Exp/Cntr=0.3,0.1

Type RM Length L Ch R = 1 ,48197.71,674.05,674.05,494.55
XS GIS Cut Line= 5
  1348176.907255   784242.505448  1347436.011126   783910.816871
  1347289.799286   783856.738535  1346945.300341   784065.040232
  1345723.864436   784823.806056
#Sta/Elev= 30
       0 1026.56   267.4 1004.62  325.47 1008.42  502.28 1003.85   639.7 1008.03
  745.16  992.93  797.14   992.5  874.23 1004.57  925.04 1002.95  993.06  990.26
 1008.71  979.92 1025.26  970.44 1048.55  969.43 1084.28   971.3 1095.98  979.17
 1326.38  998.94 1452.34  999.07 1487.44  994.69 1545.55 1002.55 1729.47 1011.03
  1776.7 1006.23 1868.14  988.24  1950.1 1009.51 2033.15 1017.19 2239.82  1015.4
 2492.14 1006.24 2634.15 1006.59 2738.33  998.52  2757.2   991.2 2808.15  999.72
#Mann= 3 , 0 , 0
       0      .1       0 1008.71    .047       0 1095.98     .11       0
#XS Ineff= 2 , 0
          874.86 1007.88 1269.86         1008.17
Permanent Ineff=
       F       F
Bank Sta=1008.71,1095.98
Exp/Cntr=0.3,0.1

Type RM Length L Ch R = 1 ,47523.66,426.36,426.36,611.32
XS GIS Cut Line= 5
  1348575.930743   783908.188391  1347407.618678   783609.819495
   1347260.20095   783228.050151  1346936.175989   782993.043047
  1345750.458484   783655.335655
#Sta/Elev= 30
       0  1017.8  271.91  992.56  354.54  995.59  398.96 1005.38  416.19 1005.63
  470.23 1020.32  516.78 1022.44  671.42 1010.53  727.51 1002.71  788.94 1005.48
  978.91  999.87 1120.49  999.98 1266.52  982.26 1323.59  980.66 1356.09  974.09
 1382.52  966.15 1453.41  967.48 1474.48  974.42 1514.32  984.29 1723.75  986.87
 1819.01  992.93 2073.51  986.34 2210.75  997.64 2336.44  983.74 2729.31  993.18
 2878.55 1002.37 3155.23 1052.84 3220.43 1059.18 3300.91 1061.54 3373.47 1069.42
#Mann= 3 , 0 , 0
       0     .11       0 1356.09    .047       0 1474.48     .11       0
Bank Sta=1356.09,1474.48
Exp/Cntr=0.3,0.1

Type RM Length L Ch R = 1 ,47097.3 ,472.88,472.88,736.4
XS GIS Cut Line= 2
  1348043.557751   783256.535783  1346907.690229   782918.268007
#Sta/Elev= 30
       0 1070.02   15.54 1068.22   31.21 1063.94   46.65 1061.95    82.5 1053.98
  226.76 1012.69  266.41  998.19  295.56     992  334.74  980.99  353.14  973.43
  371.07  966.29  376.16  965.63  395.57  966.47  419.37  965.35  448.31  965.94
  466.64  972.04  508.31  977.76  534.24  984.01  549.62  988.95  579.15  994.91
  608.59  999.27  671.74 1002.61  735.33 1000.14  784.17  996.36  824.28  997.26
  934.53 1004.88  998.53 1004.92  1052.8 1002.72 1119.09   995.9 1185.17  990.59
#Mann= 3 , 0 , 0
       0     .12       0  353.14    .047       0  466.64     .12       0
Bank Sta=353.14,466.64
Exp/Cntr=0.3,0.1

Type RM Length L Ch R = 1 ,46624.41,521.23,521.23,503.48
XS GIS Cut Line= 2
   1347768.99391    782478.58903  1347479.931382   782942.130663
#Sta/Elev= 30
       0  1009.2   30.73 1008.51   51.57 1012.35   63.58 1013.65   68.18 1013.65
   89.25 1015.35   99.59 1015.34  115.68 1013.71  131.13 1011.36  159.54  999.98
  189.73  986.75  201.46   984.1  216.44  978.43  228.11  975.86  243.72  969.56
  245.72   969.1  251.01  963.31   265.6  964.34     287  963.31  309.89  964.31
  328.72  969.73  329.66  970.24  342.33  972.71  347.11  972.79  361.45   974.4
  385.81  978.17  413.61  981.29   471.7  991.18  532.94   998.3  546.29   999.2
#Mann= 3 , 0 , 0
       0     .12       0  243.72    .047       0  328.72     .12       0
Bank Sta=243.72,328.72
Exp/Cntr=0.3,0.1

Type RM Length L Ch R = 1 ,46103.19,547.57,547.57,324.74
XS GIS Cut Line= 2
  1347331.493878   782298.901478  1346925.437173   782831.024358
#Sta/Elev= 30
       0 1001.36    65.3  989.75  106.97  983.93  139.56  982.71  239.31  973.14
  278.45  971.86  280.75  971.06  298.05  961.05  301.62  959.94  306.26  958.91
   313.4  959.67  336.51  958.67  359.95  959.67  366.87  962.49  372.45  970.01
  387.12  973.02  393.29  979.78  409.38  987.72  425.37 1001.71  433.64 1005.28
  437.52 1006.15  451.15 1019.79  474.66 1025.68  506.44 1030.63  533.78 1028.05
   555.1 1024.64   571.4 1021.37  586.08 1017.27  600.73  1015.2  669.36  999.83
#Mann= 3 , 0 , 0
       0     .12       0  280.75    .047       0  372.45     .12       0
Bank Sta=280.75,372.45
Exp/Cntr=0.3,0.1

Type RM Length L Ch R = 1 ,45555.62,409.77,409.77,414.55
XS GIS Cut Line= 2
  1347308.056438   782137.443174  1346732.535541   782028.068198
#Sta/Elev= 30
       0 1001.92   20.44  998.69    29.1   996.8   63.65  990.74    72.1  988.95
   87.62  987.53  120.45  981.64  145.29   980.8  160.64  978.82  168.36  978.64
  190.81  975.57  202.75  973.59  249.47   967.3  284.09  958.42  305.76  959.13
  328.64  958.13  351.92  959.13  361.44  968.45  365.61  971.74  379.28  981.32
  381.71  985.95  391.75  992.71  404.12 1000.01  412.57 1005.63  431.69 1012.37
  461.44 1021.33  489.48 1027.14  506.74 1028.28  524.97  1030.1  585.82 1037.96
#Mann= 3 , 0 , 0
       0     .12       0  249.47    .047       0  361.44     .12       0
Bank Sta=249.47,361.44
Exp/Cntr=0.3,0.1

Type RM Length L Ch R = 1 ,45145.86,615.32,615.32,945.47
XS GIS Cut Line= 2
   1347547.63967   781754.630629  1346886.181365   781645.255653
#Sta/Elev= 30
       0 1001.48   14.08  997.72   63.98     988   77.12  986.31  110.05  991.31
  148.47  991.68  174.35  995.61  199.32  993.52  215.46  993.87  233.12  995.67
  240.87  997.53  248.67  996.31  256.16  993.67  266.43   992.3  288.49  991.78
  309.12  989.57  352.24  981.42  393.72  971.14  418.83  963.58  428.86  957.74
  454.64  958.73  477.75  957.73  500.99  958.68  526.73  966.45  532.13  974.33
  581.19  993.42  605.08  996.63   617.9  996.83  639.97 1000.35  670.44  998.68
#Mann= 3 , 0 , 0
       0     .11       0  418.83    .047       0  526.73     .11       0
Bank Sta=418.83,526.73
Exp/Cntr=0.3,0.1

Type RM Length L Ch R = 1 ,44530.54,650.84,650.84,851.97
XS GIS Cut Line= 2
   1347000.26879   780739.111524  1346901.172213   781590.816101
#Sta/Elev= 30
       0 1056.59    52.9 1060.93   93.12 1062.11  152.88 1056.77  192.16 1046.31
  217.65 1043.44   239.6 1032.74  264.37 1022.52  281.37 1010.97   303.9  989.14
   305.3  986.33  321.96  969.78  322.88  964.36   323.4  958.87  323.89   955.9
  347.52  956.92  368.38  955.92  403.04  956.77  417.67  965.75  420.38  965.41
  421.15  967.76  456.53  964.99  468.08  966.04  509.89  966.92  555.89  969.21
  577.98   969.1   633.5  971.97  708.13  979.86  742.58  981.22  857.45  991.89
#Mann= 3 , 0 , 0
       0     .11       0  322.88    .047       0  417.67     .11       0
Bank Sta=322.88,417.67
Exp/Cntr=0.3,0.1

Type RM Length L Ch R = 1 ,43879.7 ,595.92,595.92,513.47
XS GIS Cut Line= 2
  1346364.647413   781329.293925  1346826.285557   781744.213989
#Sta/Elev= 30
       0 1012.65   32.17 1010.27   42.22 1011.03   98.84 1008.03  124.84 1004.34
  137.86 1003.94  149.44 1002.53  165.21 1001.37  176.98  998.08  185.63  996.77
  219.55  994.05   255.4  989.09  299.98  979.66  319.82  974.97  351.27  967.23
  362.06  963.85  370.23  964.19  375.12  962.95  381.27  956.05  387.65  956.43
  410.48  955.45   435.1  956.37  456.49  955.86  469.52  966.75  486.95  971.85
  500.62  978.22  543.97  993.35   573.3 1000.65  592.21 1004.72   620.7 1008.95
#Mann= 3 , 0 , 0
       0     .11       0  370.23    .047       0  469.52     .11       0
Bank Sta=370.23,469.52
Exp/Cntr=0.3,0.1

Type RM Length L Ch R = 1 ,43283.79,498.24,498.24,360
XS GIS Cut Line= 2
  1346134.403957   781769.658085  1346344.514677    782228.58903
#Sta/Elev= 30
       0  984.09   36.31   982.2   88.93  976.88   97.43  975.61   124.8  972.86
  136.97  971.08  167.88  969.51  183.98  969.27  193.18  963.87  214.41  954.81
  216.17   955.1  239.21   954.2  262.26  955.09  275.39  953.92  281.17  957.05
  287.69  962.12  293.97  965.04   306.7  968.33  311.53  970.57  323.62  980.93
  336.62  990.85  360.19 1008.19  371.77 1017.56  376.67 1023.38  401.42 1044.54
  437.41 1056.72  467.01 1065.56  471.53 1066.28  479.26 1068.33  504.74 1073.93
#Mann= 3 , 0 , 0
       0     .11       0  193.18    .047       0  287.69     .11       0
Bank Sta=193.18,287.69
Exp/Cntr=0.3,0.1

Type RM Length L Ch R = 1 ,42785.54,712.81,712.81,434.59
XS GIS Cut Line= 2
   1345821.60818   781809.849189  1345706.394612   782251.079398
#Sta/Elev= 30
       0  977.24   10.09  976.26   60.39  975.37   72.09  975.43   86.17  974.61
  112.46  975.56  153.94  969.11  158.46  969.33  186.44  969.05  209.28  971.61
  216.74  971.26  219.45  970.91  227.89  968.23  240.62  960.67  250.45  954.07
  259.06  952.51  281.49  951.51  309.34  952.89  317.38  957.94  329.19  964.42
  334.19  965.21  344.15  967.86  356.86  972.88  380.41  990.82  389.28   997.7
  398.95 1005.78   406.6 1011.42  427.22 1030.02  432.74 1033.62  456.02 1050.39
#Mann= 3 , 0 , 0
       0     .11       0  240.62    .047       0  329.19     .11       0
Bank Sta=240.62,329.19
Exp/Cntr=0.3,0.1

Type RM Length L Ch R = 1 ,42072.73,675.7,675.7,351.29
XS GIS Cut Line= 3
  1345795.035508   781593.172325  1345177.848052   781551.505637
  1344614.875379    782143.51767
#Sta/Elev= 30
       0  977.52  214.32  968.47  386.22  967.83  413.88  953.18  418.51  955.78
  440.79   950.5  464.41  956.53  473.17  951.94   488.7  967.26  536.62 1001.63
  555.97 1011.39  567.18 1012.61  593.77  1009.3  618.59  998.93  677.19  996.17
   705.4  986.32  777.31  988.27  809.88  995.04  864.78   992.9   907.6  979.52
  934.46  989.46  973.51  998.96 1046.19 1008.81 1078.48 1007.84 1121.95 1010.94
 1149.82 1009.03 1187.88 1013.97 1285.57 1016.78 1339.53 1008.04 1435.55 1000.93
#Mann= 3 , 0 , 0
       0     .11       0  386.22    .047       0   488.7     .11       0
#XS Ineff= 2 , 0
                          579.76         1016.07
Permanent Ineff=
       F       F
Bank Sta=386.22,488.7
Exp/Cntr=0.3,0.1
