HEC-RAS study North Little Hunting Creek.prj: North Little Hunting Creek Limited Detail Study

--- North Little Hunting Creek.g01 (geometry) --- (continued)

Type RM Length L Ch R = 1,79939,562,562,562
BEGIN DESCRIPTION:
North Hunting Creek 141.0
END DESCRIPTION:
XS GIS Cut Line= 4
      1453853.87       867839.50      1453742.04       867806.37
      1453601.23       867769.09      1453427.34       867771.16
#Sta/Elev= 30
  4818.8  992.32  4820.2  992.25  4839.5  987.18  4862.6  982.28  4874.2  981.56
  4883.3  979.69  4895.9  977.75  4911.1  976.20  4915.2  976.15  4935.2  973.03
  4953.0  973.01  4970.7  970.84  4982.5  962.30  4983.5  960.30  5016.5  960.30
  5017.5  962.30  5022.2  963.04  5026.6  962.30  5028.4  964.63  5028.9  965.48
  5030.7  966.04  5054.3  970.85  5062.6  971.53  5080.9  971.66  5099.4  973.06
  5127.6  976.16  5158.4  980.70  5199.2  987.97  5234.5  996.12  5255.0  999.93
#Mann=3,-1,0
  4818.8    0.12       0  4982.5    0.04       0  5017.5    0.12       0
Bank Sta=4982.5,5017.5
XS Rating Curve= 0
Exp/Cntr=0.3,0.1

Type RM Length L Ch R = 1,79377,607,607,607
BEGIN DESCRIPTION:
North Hunting Creek 140.0
END DESCRIPTION:
XS GIS Cut Line= 2
      1454079.54       867427.43      1453816.59       867195.53
#Sta/Elev= 30
  4799.1  980.19  4810.2  979.48  4820.0  978.66  4841.6  977.38  4852.0  976.88
  4862.7  976.70  4873.3  976.17  4883.2  975.25  4893.6  974.75  4903.8  973.86
  4924.7  971.69  4935.6  971.12  4945.3  970.84  4948.0  970.67  4963.9  969.67
  4965.2  969.49  4982.0  962.91  4982.5  961.06  4983.5  959.06  5016.5  959.06
  5017.5  961.06  5020.8  965.36  5048.7  972.32  5058.0  975.03  5071.6  980.22
  5080.0  982.48  5088.7  984.68  5102.9  987.56  5133.1  991.70  5149.7  994.23
#Mann=4,-1,0
  4799.1    0.06       0  4948.0    0.12       0  4982.5    0.04       0
  5017.5    0.12       0
Bank Sta=4982.5,5017.5
XS Rating Curve= 0
Exp/Cntr=0.3,0.1

Type RM Length L Ch R = 1,78770,562,562,562
BEGIN DESCRIPTION:
North Hunting Creek 139.0
END DESCRIPTION:
XS GIS Cut Line= 4
      1454388.05       866812.45      1454284.55       866804.17
      1454195.51       866802.10      1453996.72       866858.01
#Sta/Elev= 30
  4861.3  995.54  4866.2  994.14  4888.0  989.33  4892.2  988.11  4908.6  982.62
  4928.8  976.37  4933.9  974.42  4945.5  971.13  4965.1  967.65  4982.5  959.88
  4983.5  957.88  5016.5  957.88  5017.5  959.88  5025.8  968.39  5050.6  969.98
  5067.6  971.80  5072.3  972.18  5087.4  973.96  5102.6  975.49  5113.8  977.03
  5141.5  980.07  5155.3  981.19  5160.5  981.72  5168.8  982.80  5183.5  983.64
  5199.3  984.79  5212.7  985.18  5224.0  985.65  5244.6  987.69  5260.7  989.15
#Mann=3,-1,0
  4861.3    0.09       0  4982.5    0.04       0  5017.5    0.09       0
Bank Sta=4982.5,5017.5
XS Rating Curve= 0
Exp/Cntr=0.3,0.1

Type RM Length L Ch R = 1,78208,533,533,533
BEGIN DESCRIPTION:
North Hunting Creek 138.0
END DESCRIPTION:
XS GIS Cut Line= 3
      1454439.84       866352.77      1454344.59       866284.44
      1454238.98       866207.82
#Sta/Elev= 24
  4848.3  981.24  4868.7  978.37  4873.5  977.59  4881.6  976.08  4894.6  974.12
  4903.5  972.46  4915.1  970.57  4924.0  969.40  4926.4  969.25  4936.0  968.38
  4945.5  968.13  4957.6  966.97  4977.8  964.19  4982.5  958.43  4983.5  956.43
  5016.5  956.43  5017.5  958.43  5041.5  985.76  5050.7  989.83  5063.3  995.96
  5073.2 1001.99  5077.2 1003.89  5085.8 1007.69  5096.0 1010.04
#Mann=3,-1,0
  4848.3    0.09       0  4982.5    0.04       0  5017.5    0.09       0
Bank Sta=4982.5,5017.5
XS Rating Curve= 0
Exp/Cntr=0.3,0.1

Type RM Length L Ch R = 1,77675,596,596,596
BEGIN DESCRIPTION:
North Hunting Creek 137.0
END DESCRIPTION:
XS GIS Cut Line= 4
      1454909.88       865961.42      1454758.72       865932.43
      1454642.77       865853.75      1454522.69       865874.45
#Sta/Elev= 30
  4752.3  990.02  4799.1  984.07  4837.3  979.89  4852.8  975.68  4874.1  970.68
  4879.1  969.87  4884.2  969.63  4904.8  966.16  4910.1  965.61  4938.4  964.09
  4949.5  962.74  4978.1  961.13  4982.5  957.15  4983.5  955.15  5016.5  955.15
  5017.5  957.15  5018.8  959.83  5026.6  962.80  5046.0  968.00  5049.2  968.37
  5053.4  969.58  5078.4  975.05  5084.0  976.70  5100.0  980.35  5103.2  980.82
  5106.7  981.96  5113.5  983.34  5142.5  991.02  5152.6  992.12  5168.2  994.82
#Mann=3,-1,0
  4752.3    0.09       0  4982.5    0.04       0  5017.5    0.09       0
Bank Sta=4982.5,5017.5
XS Rating Curve= 0
Exp/Cntr=0.3,0.1

Type RM Length L Ch R = 1,77079,579,579,579
BEGIN DESCRIPTION:
North Hunting Creek 136.0
END DESCRIPTION:
XS GIS Cut Line= 3
      1455197.70       865507.94      1455106.59       865449.97
      1454951.26       865352.63
#Sta/Elev= 30
  4817.9  987.69  4822.4  987.63  4825.1  987.18  4835.5  985.85  4839.8  985.06
  4846.0  983.48  4853.1  982.18  4864.2  979.80  4866.7  979.08  4880.6  976.26
  4888.5  975.78  4902.4  971.16  4910.3  969.08  4930.3  964.60  4941.8  963.24
  4948.3  962.75  4972.0  957.76  4974.5  956.54  4982.2  955.25  4983.2  953.25
  5016.8  953.25  5017.8  955.25  5024.6  959.91  5032.6  963.97  5047.8  969.31
  5057.2  972.92  5079.5  983.85  5096.9  991.99  5101.6  994.03  5109.2  996.62
#Mann=3,-1,0
  4817.9    0.09       0  4982.2    0.04       0  5017.8    0.09       0
Bank Sta=4982.2,5017.8
XS Rating Curve= 0
Exp/Cntr=0.3,0.1

Type RM Length L Ch R = 1,76500,593,593,593
BEGIN DESCRIPTION:
North Hunting Creek 135.0
END DESCRIPTION:
XS GIS Cut Line= 3
      1455491.76       864982.01      1455357.14       864917.81
      1455170.81       864849.49
#Sta/Elev= 30
  4798.5  975.89  4815.3  973.77  4841.4  970.78  4854.1  969.57  4860.5  968.67
  4880.2  967.42  4897.5  965.25  4909.9  963.56  4920.1  961.91  4925.1  961.39
  4926.6  961.42  4943.3  960.29  4949.1  960.27  4962.4  956.81  4964.4  956.47
  4969.0  956.00  4982.2  953.53  4983.2  951.53  5016.8  951.53  5017.8  953.53
  5027.4  962.12  5034.4  966.23  5057.3  974.98  5062.3  976.23  5074.8  980.09
  5079.7  981.43  5096.1  985.03  5109.3  987.42  5135.7  991.36  5146.1  992.71
#Mann=3,-1,0
  4798.5    0.09       0  4982.2    0.04       0  5017.8    0.09       0
Bank Sta=4982.2,5017.8
XS Rating Curve= 0
Exp/Cntr=0.3,0.1

Type RM Length L Ch R = 1,75907,487,487,487
BEGIN DESCRIPTION:
North Hunting Creek 134.0
END DESCRIPTION:
XS GIS Cut Line= 4
      1455423.44       864306.96      1455326.08       864331.82
      1455230.83       864383.59      1455143.85       864520.27
#Sta/Elev= 30
  4876.0  980.95  4882.5  979.80  4889.0  979.28  4898.0  978.12  4908.3  976.22
  4916.9  973.96  4925.4  972.03  4940.6  967.57  4943.4  966.57  4949.4  963.78
  4961.6  959.42  4972.3  953.12  4976.5  952.72  4982.2  949.84  4983.2  947.84
  5016.8  947.84  5017.8  949.84  5019.1  954.18  5028.3  956.70  5048.1  959.60
  5064.7  960.82  5080.0  961.55  5088.0  962.49  5112.6  964.67  5135.4  965.62
  5155.3  967.14  5159.7  967.58  5198.0  972.56  5235.0  976.55  5246.9  977.99
#Mann=4,-1,0
  4876.0    0.12       0  4982.2    0.04       0  5017.8    0.12       0
  5088.0    0.06       0
Bank Sta=4982.2,5017.8
XS Rating Curve= 0
Exp/Cntr=0.3,0.1

Type RM Length L Ch R = 1,75420,223,223,223
BEGIN DESCRIPTION:
North Hunting Creek 133.5
END DESCRIPTION:
XS GIS Cut Line= 4
      1455421.85       864288.77      1455337.14       864028.67
      1455362.40       863783.44      1455380.23       863698.77
#Sta/Elev= 30
  4624.0  978.21  4647.9  975.10  4674.8  970.69  4717.2  965.79  4732.8  964.71
  4737.9  963.93  4795.7  961.24  4816.8  958.67  4843.7  956.73  4864.7  952.49
  4877.5  951.53  4904.1  956.54  4923.9  957.38  4937.6  956.33  4970.5  956.92
  4972.0  956.68  4982.2  948.68  4983.2  946.68  5016.8  946.68  5017.8  948.68
  5030.1  950.63  5064.1  954.75  5087.0  955.09  5128.3  957.20  5145.3  960.59
  5166.8  962.24  5183.3  968.25  5207.3  971.91  5219.8  975.91  5230.6  978.19
#Mann=3,-1,0
  4624.0    0.08       0  4982.2    0.04       0  5017.8    0.12       0
Bank Sta=4982.2,5017.8
XS Rating Curve= 0
Exp/Cntr=0.3,0.1

Type RM Length L Ch R = 1,75197,447,447,447
BEGIN DESCRIPTION:
North Hunting Creek 133.0
END DESCRIPTION:
XS GIS Cut Line= 4
      1455439.96       864280.04      1455388.20       864155.81
      1455568.35       863977.74      1455663.60       863967.38
#Sta/Elev= 30
  4715.5  977.00  4745.3  972.59  4766.1  970.17  4786.1  966.89  4796.4  965.86
  4806.6  965.20  4812.1  964.32  4827.3  963.68  4832.6  963.00  4850.1  962.38
  4899.6  959.96  4917.7  959.70  4928.8  960.00  4943.3  959.49  4959.6  959.28
  4973.6  956.81  4982.2  947.24  4983.2  945.24  5016.8  945.24  5017.8  947.24
  5032.4  958.36  5049.9  958.26  5065.4  957.51  5082.3  954.60  5091.3  955.04
  5111.4  954.92  5117.2  957.95  5146.4  967.59  5172.8  974.75  5199.2  979.14
#Mann=3,-1,0
  4715.5    0.06       0  4982.2    0.04       0  5017.8    0.12       0
#XS Ineff=2,0
       0                 5032.40    0.00  958.36
Permanent Ineff=
       F       F
Bank Sta=4982.2,5017.8
XS Rating Curve= 0
Exp/Cntr=0.3,0.1

Type RM Length L Ch R = 1,74750,637,637,637
BEGIN DESCRIPTION:
North Hunting Creek 132.0
END DESCRIPTION:
XS GIS Cut Line= 4
      1455854.10       864362.89      1455845.81       864284.19
      1455827.18       864201.37      1455758.84       864041.92
#Sta/Elev= 30
  4900.5 1005.00  4906.6 1003.01  4914.5  999.59  4919.1  997.72  4930.1  990.80
  4931.6  989.94  4941.3  983.35  4944.4  980.53  4950.5  976.21  4957.4  970.72
  4960.9  968.05  4965.3  963.95  4975.7  952.79  4979.6  949.15  4982.2  944.86
  4983.2  942.86  5016.8  942.86  5017.8  944.86  5046.4  955.54  5048.8  955.86
  5050.2  955.98  5099.7  956.60  5128.8  960.88  5139.8  962.73  5165.5  963.61
  5171.4  964.19  5177.4  965.04  5224.5  969.14  5233.7  970.96  5238.0  971.45
#Mann=3,-1,0
  4900.5    0.12       0  4982.2    0.04       0  5017.8    0.12       0
Bank Sta=4982.2,5017.8
XS Rating Curve= 0
Exp/Cntr=0.3,0.1

Type RM Length L Ch R = 1,74113,347,347,347
BEGIN DESCRIPTION:
North Hunting Creek 131.0
END DESCRIPTION:
XS GIS Cut Line= 4
      1456440.09       864101.97      1456394.54       863967.39
      1456348.98       863886.63      1456239.24       863735.47
#Sta/Elev= 30
  4801.2  965.67  4811.6  964.69  4832.2  964.60  4838.2  963.43  4856.7  961.04
  4887.8  955.42  4901.1  953.46  4937.4  950.48  4942.6  950.72  4945.8  949.24
  4954.3  946.94  4967.2  944.04  4982.2  941.69  4983.2  939.69  5016.8  939.69
  5017.8  941.69  5025.0  949.38  5026.7  949.15  5034.5  950.04  5044.3  950.41
  5053.4  952.71  5086.7  958.70  5089.6  959.84  5110.6  963.64  5125.8  965.35
  5148.0  965.87  5169.4  967.60  5174.6  966.97  5190.5  968.19  5222.8  969.10
#Mann=3,-1,0
  4801.2    0.12       0  4982.2    0.04       0  5017.8    0.12       0
Bank Sta=4982.2,5017.8
XS Rating Curve= 0
Exp/Cntr=0.3,0.1

Type RM Length L Ch R = 1,73766,247,247,247
BEGIN DESCRIPTION:
North Little Hunting Creek 130.5
END DESCRIPTION:
XS GIS Cut Line= 4
      1456561.01       864093.04      1456676.05       863986.60
      1456668.53       863746.87      1456726.59       863624.30
#Sta/Elev= 30
  4626.9  966.06  4645.4  964.59  4683.4  963.01  4709.5  962.72  4742.5  961.36
  4757.9  960.21  4773.0  960.42  4779.1  960.12  4827.6  955.24  4864.2  952.09
  4883.6  951.68  4897.6  950.86  4921.6  948.52  4930.9  948.24  4950.0  946.13
  4952.3  946.27  4960.8  945.33  4965.3  944.37  4972.7  944.04  4982.2  940.06
  4983.2  938.06  5016.8  938.06  5017.8  940.06  5023.5  943.91  5051.9  951.89
  5068.2  954.07  5077.2  955.86  5100.9  958.22  5128.7  964.19  5159.1  968.46
#Mann=3,-1,0
  4626.9    0.12       0  4982.2    0.04       0  5017.8    0.12       0
Bank Sta=4982.2,5017.8
XS Rating Curve= 0
Exp/Cntr=0.3,0.1

Type RM Length L Ch R = 1,73519,537,537,537
BEGIN DESCRIPTION:
North Hunting Creek 130.0
END DESCRIPTION:
XS GIS Cut Line= 4
      1456924.62       863957.00      1456916.34       863872.14
      1456910.13       863778.96      1456881.13       863648.49
#Sta/Elev= 30
  4840.0  976.18  4848.9  975.81  4857.8  975.04  4870.3  972.31  4878.1  969.12
  4883.6  967.59  4902.1  957.97  4905.7  956.95  4920.4  953.22  4926.9  951.35
  4951.2  946.01  4961.9  945.40  4968.7  944.71  4982.2  938.70  4983.2  936.70
  5016.8  936.70  5017.8  938.70  5018.7  943.98  5047.8  951.68  5059.1  954.36
  5081.6  962.75  5089.0  963.33  5093.5  964.38  5098.0  965.58  5113.3  969.03
  5118.6  969.59  5126.5  970.22  5136.6  970.64  5145.9  971.26  5152.3  972.48
#Mann=3,-1,0
  4840.0    0.12       0  4982.2    0.04       0  5017.8    0.12       0
Bank Sta=4982.2,5017.8
XS Rating Curve= 0
Exp/Cntr=0.3,0.1

Type RM Length L Ch R = 1,72982,650,650,650
BEGIN DESCRIPTION:
North Hunting Creek 129.0
END DESCRIPTION:
XS GIS Cut Line= 3
      1457235.22       863511.84      1457156.53       863489.07
      1456945.36       863491.14
#Sta/Elev= 28
  4855.2  962.06  4857.0  961.97  4876.4  960.05  4881.6  959.15  4904.4  954.58
  4909.1  953.05  4913.3  952.18  4929.0  946.56  4932.3  946.32  4937.1  945.92
  4948.7  945.05  4968.0  944.07  4970.9  943.50  4977.3  937.12  4978.5  935.12
  5021.5  935.12  5022.7  937.12  5036.9  942.85  5041.1  943.79  5081.6  952.63
  5100.4  958.02  5104.2  959.28  5107.3  960.71  5111.6  962.21  5133.1  970.35
  5145.3  974.27  5145.4  974.32  5148.3  975.18
#Mann=3,-1,0
  4855.2    0.12       0  4977.3    0.04       0  5022.7    0.12       0
Bank Sta=4977.3,5022.7
XS Rating Curve= 0
Exp/Cntr=0.3,0.1

Type RM Length L Ch R = 1,72332,572,572,572
BEGIN DESCRIPTION:
North Hunting Creek 128.0
END DESCRIPTION:
XS GIS Cut Line= 4
      1457510.61       863275.81      1457518.90       863147.41
      1457440.21       862992.11      1457394.65       862936.19
#Sta/Elev= 30
  4709.1  963.78  4719.2  963.41  4727.1  962.25  4733.3  960.98  4757.3  959.29
  4760.0  958.67  4767.7  957.28  4808.2  952.15  4816.1  950.99  4820.4  950.04
  4837.8  948.60  4842.0  948.44  4851.3  947.47  4869.0  946.40  4878.7  946.10
  4887.8  946.00  4893.4  945.75  4933.0  943.15  4947.9  942.85  4952.1  943.14
  4981.1  932.79  4982.1  930.79  5017.9  930.79  5018.9  932.79  5022.9  942.02
  5023.7  942.53  5027.1  945.32  5058.2  971.56  5073.1  980.22  5084.0  986.05
#Mann=3,-1,0
  4709.1    0.08       0  4981.1    0.04       0  5018.9    0.12       0
Bank Sta=4981.1,5018.9
XS Rating Curve= 0
Exp/Cntr=0.3,0.1

Type RM Length L Ch R = 1,71760,538,538,538
BEGIN DESCRIPTION:
North Hunting Creek 127.0
END DESCRIPTION:
XS GIS Cut Line= 4
      1458082.11       863045.92      1458075.90       862919.64
      1457941.31       862735.35      1457895.75       862650.44
#Sta/Elev= 30
  4666.3  963.72  4699.9  960.93  4709.4  959.93  4729.5  957.02  4742.6  955.52
  4760.7  951.94  4780.2  950.25  4787.6  949.71  4792.7  949.64  4838.3  947.12
  4903.3  942.68  4908.2  942.67  4918.2  942.01  4937.7  941.57  4945.7  941.08
  4964.0  939.28  4967.0  938.75  4981.1  931.10  4982.1  929.10  5017.9  929.10
  5018.9  931.10  5020.9  936.78  5037.7  946.00  5042.8  948.27  5067.4  961.46
  5074.5  965.07  5085.6  966.58  5094.5  968.21  5112.6  970.41  5117.3  971.19
#Mann=3,-1,0
  4666.3    0.08       0  4981.1    0.04       0  5018.9    0.12       0
Bank Sta=4981.1,5018.9
XS Rating Curve= 0
Exp/Cntr=0.3,0.1

Type RM Length L Ch R = 1,71222,628,628,628
BEGIN DESCRIPTION:
North Hunting Creek 126.0
END DESCRIPTION:
XS GIS Cut Line= 4
      1458409.32       862319.13      1458305.74       862368.85
      1458175.29       862397.84      1457951.63       862517.95
#Sta/Elev= 30
  4861.4  978.14  4878.6  974.60  4891.8  970.77  4905.1  965.87  4922.6  960.31
  4957.2  944.59  4962.9  941.46  4979.4  936.48  4981.1  929.31  4982.1  927.31
  5017.9  927.31  5018.9  929.31  5021.1  934.81  5028.3  937.83  5031.8  938.33
  5045.1  939.65  5063.1  940.82  5081.1  939.03  5099.7  940.59  5118.3  943.01
  5135.5  947.10  5142.6  947.53  5169.8  952.08  5206.2  956.24  5225.5  957.69
  5243.7  959.95  5254.0  960.17  5291.9  963.50  5331.4  965.86  5363.8  969.15
#Mann=3,-1,0
  4861.4    0.12       0  4981.1    0.04       0  5018.9    0.12       0
Bank Sta=4981.1,5018.9
XS Rating Curve= 0
Exp/Cntr=0.3,0.1

Type RM Length L Ch R = 1,70594,551,551,551
BEGIN DESCRIPTION:
North Hunting Creek 125.0
END DESCRIPTION:
XS GIS Cut Line= 4
      1458318.19       861737.29      1458169.08       861772.50
      1457740.46       861956.79      1457659.67       861989.93
#Sta/Elev= 30
  4835.7  970.21  4842.9  968.97  4886.3  943.17  4897.5  939.93  4926.5  937.49
  4956.7  937.99  4976.5  930.16  4980.3  930.00  4981.1  927.04  4982.1  925.04
  5017.9  925.04  5018.9  927.04  5019.1  933.18  5028.3  939.37  5034.0  940.41
  5065.4  939.16  5085.6  940.61  5111.6  941.57  5147.4  941.91  5180.9  939.18
  5192.5  939.27  5218.1  938.22  5254.4  939.17  5290.1  941.51  5336.8  941.16
  5394.7  939.45  5428.4  939.99  5446.6  941.22  5478.0  951.25  5542.8  980.47
#Mann=3,-1,0
  4835.7    0.12       0  4981.1    0.04       0  5018.9    0.12       0
#XS Ineff=2,0
       0                 5040.10    0.00  940.43
Permanent Ineff=
       F       F
Bank Sta=4981.1,5018.9
XS Rating Curve= 0
Exp/Cntr=0.3,0.1

Type RM Length L Ch R = 1,70043,699,699,699
BEGIN DESCRIPTION:
North Hunting Creek 124.0
END DESCRIPTION:
XS GIS Cut Line= 4
      1458181.85       861550.62      1457788.25       861438.44
      1457516.67       861617.52      1457418.27       861708.05
#Sta/Elev= 30
  4486.8  958.01  4509.2  956.29  4577.5  949.21  4650.0  951.70  4731.4  947.63
  4750.3  945.57  4774.0  944.23  4791.7  941.81  4817.6  941.37  4852.5  939.00
  4896.6  938.10  4911.5  937.10  4942.4  938.61  4960.3  937.33  4981.1  925.67
  4982.1  923.67  5017.9  923.67  5018.9  925.67  5020.9  928.23  5033.0  931.63
  5071.4  938.35  5081.5  938.77  5134.0  937.12  5182.6  937.53  5203.1  937.04
  5241.4  938.32  5260.3  942.04  5277.2  947.70  5322.9  967.63  5355.1  979.91
#Mann=3,-1,0
  4486.8    0.12       0  4981.1    0.04       0  5018.9    0.12       0
Bank Sta=4981.1,5018.9
XS Rating Curve= 0
Exp/Cntr=0.3,0.1

Type RM Length L Ch R = 1,69344,238,238,238
BEGIN DESCRIPTION:
North Hunting Creek 123.5
END DESCRIPTION:
XS GIS Cut Line= 4
      1458189.14       861542.03      1457809.23       861413.56
      1457858.79       861213.49      1457906.52       861123.53
#Sta/Elev= 30
  4420.5  957.94  4452.2  955.10  4475.6  952.11  4503.0  949.81  4533.1  949.63
  4588.4  951.34  4643.9  950.39  4671.8  948.94  4708.5  945.09  4736.2  943.87
  4749.2  942.00  4792.0  938.75  4870.6  936.27  4875.0  936.59  4903.2  935.23
  4940.4  934.71  4953.3  936.35  4977.9  930.60  4979.0  929.09  4979.3  924.63
  4979.5  924.62  4980.5  922.62  5019.5  922.62  5020.5  924.62  5029.2  930.94
  5033.9  932.83  5073.7  945.30  5091.1  952.64  5111.3  957.97  5129.5  961.61
#Mann=3,-1,0
  4420.5    0.12       0  4979.5    0.04       0  5020.5    0.12       0
Bank Sta=4979.5,5020.5
XS Rating Curve= 0
Exp/Cntr=0.3,0.1

Type RM Length L Ch R = 1,69106,647,647,647
BEGIN DESCRIPTION:
North Hunting Creek 123.0
END DESCRIPTION:
XS GIS Cut Line= 4
      1458191.84       861536.42      1458111.10       861443.27
      1458067.62       861227.92      1457997.20       861105.72
#Sta/Elev= 30
  4717.3  957.74  4762.6  952.41  4772.2  950.84  4781.9  950.75  4793.9  948.79
  4844.3  945.89  4907.9  940.20  4916.3  939.88  4932.1  937.51  4952.2  935.61
  4955.4  935.77  4957.5  933.50  4963.2  928.72  4969.8  924.14  4979.5  924.13
  4980.5  922.13  5019.5  922.13  5020.5  924.13  5022.5  924.14  5023.3  927.99
  5028.9  934.87  5038.6  932.24  5048.9  932.32  5054.6  932.93  5077.1  936.92
  5089.4  940.69  5100.4  943.42  5133.1  950.31  5180.0  957.72  5201.3  959.96
#Mann=3,-1,0
  4717.3    0.12       0  4979.5    0.04       0  5020.5    0.08       0
Bank Sta=4979.5,5020.5
XS Rating Curve= 0
Exp/Cntr=0.3,0.1

Type RM Length L Ch R = 1,68459,669,669,669
BEGIN DESCRIPTION:
North Hunting Creek 122.0
END DESCRIPTION:
XS GIS Cut Line= 4
      1458705.38       861437.10      1458713.66       861221.71
      1458680.53       861037.42      1458618.40       860873.82
#Sta/Elev= 30
  4755.6  955.83  4763.3  954.40  4803.9  945.78  4829.0  939.96  4853.7  938.23
  4866.5  937.03  4903.2  935.73  4933.3  932.91  4972.1  925.46  4975.7  923.36
  4979.5  923.36  4980.5  921.36  5019.5  921.36  5020.5  923.36  5025.5  923.45
  5040.9  933.85  5049.2  933.32  5068.4  933.30  5082.6  932.88  5096.9  933.04
  5113.1  933.56  5125.5  934.43  5142.6  934.94  5180.7  937.11  5218.5  938.58
  5284.6  942.42  5297.2  944.18  5323.7  946.80  5328.1  947.00  5333.4  948.13
#Mann=3,-1,0
  4755.6    0.12       0  4979.5    0.04       0  5020.5    0.06       0
Bank Sta=4979.5,5020.5
XS Rating Curve= 0
Exp/Cntr=0.3,0.1

Type RM Length L Ch R = 1,67790,619,619,619
BEGIN DESCRIPTION:
North Hunting Creek 121.0
END DESCRIPTION:
XS GIS Cut Line= 4
      1459405.26       861219.66      1459394.90       861089.19
      1459094.66       860724.75      1458966.28       860631.58
#Sta/Elev= 30
  4743.1  954.55  4768.6  951.07  4797.2  945.19  4832.5  940.16  4862.3  936.52
  4909.9  931.80  4923.9  931.94  4934.4  933.62  4963.6  922.55  4979.5  922.55
  4980.5  920.55  5019.5  920.55  5020.5  922.55  5024.7  922.59  5025.7  925.27
  5032.8  931.71  5040.8  931.23  5051.1  932.73  5063.4  933.50  5100.6  933.12
  5122.7  932.24  5179.6  932.57  5199.9  931.33  5209.8  931.99  5250.0  932.60
  5286.9  933.92  5312.3  934.04  5363.7  937.02  5422.0  944.59  5504.8  950.22
#Mann=3,-1,0
  4743.1    0.12       0  4979.5    0.04       0  5020.5    0.12       0
Bank Sta=4979.5,5020.5
XS Rating Curve= 0
Exp/Cntr=0.3,0.1

Type RM Length L Ch R = 1,67171,395,395,395
BEGIN DESCRIPTION:
North Hunting Creek 120.0
END DESCRIPTION:
XS GIS Cut Line= 4
      1459871.13       860586.01      1459788.33       860552.89
      1459566.77       860465.92      1459405.23       860399.65
#Sta/Elev= 30
  4835.3  960.27  4838.4  959.92  4876.8  946.58  4908.5  936.51  4917.9  932.49
  4929.2  928.85  4937.5  928.48  4946.7  928.50  4967.7  929.32  4978.5  928.91
  4979.5  921.74  4980.5  919.74  5019.5  919.74  5020.5  921.74  5024.0  921.75
  5030.7  926.89  5034.3  931.57  5043.8  930.98  5050.0  931.27  5055.6  931.93
  5071.1  931.98  5113.6  931.01  5137.0  930.95  5173.0  933.24  5199.6  934.58
  5211.3  933.89  5235.6  935.64  5259.3  938.59  5288.8  940.38  5337.1  944.42
#Mann=3,-1,0
  4835.3    0.12       0  4979.5    0.04       0  5020.5    0.12       0
Bank Sta=4979.5,5020.5
XS Rating Curve= 0
Exp/Cntr=0.3,0.1

Type RM Length L Ch R = 1,66776,338,338,338
BEGIN DESCRIPTION:
North Hunting Creek 119.5
END DESCRIPTION:
XS GIS Cut Line= 4
      1460034.69       860327.11      1459927.15       860248.69
      1459799.48       860121.02      1459714.37       860026.95
#Sta/Elev= 30
  4726.4  948.28  4732.4  947.93  4796.1  941.24  4801.8  940.05  4809.0  938.11
  4849.2  931.69  4870.4  930.77  4874.4  930.22  4879.5  930.28  4888.3  929.80
  4896.5  930.31  4916.2  930.52  4927.9  931.01  4938.7  930.81  4955.8  927.92
  4966.9  921.33  4979.5  921.33  4980.5  919.33  5019.5  919.33  5020.5  921.33
  5035.9  921.33  5036.5  927.04  5046.0  931.80  5050.0  932.25  5057.0  932.23
  5109.4  947.81  5129.3  952.24  5136.5  955.42  5157.3  957.81  5166.9  959.28
#Mann=3,-1,0
  4726.4    0.12       0  4979.5    0.04       0  5020.5    0.12       0
Bank Sta=4979.5,5020.5
XS Rating Curve= 0
Exp/Cntr=0.3,0.1

Type RM Length L Ch R = 1,66438,490,490,490
BEGIN DESCRIPTION:
North Hunting Creek 119.0
END DESCRIPTION:
XS GIS Cut Line= 4
      1460181.76       860260.89      1460245.94       860047.65
      1460034.73       859898.56      1459881.50       859815.73
#Sta/Elev= 30
  4568.6  943.68  4589.3  942.51  4603.6  941.08  4652.5  937.63  4715.9  933.80
  4801.1  931.95  4839.9  930.12  4879.4  931.68  4891.8  930.27  4898.9  928.96
  4911.2  928.62  4939.1  929.42  4971.8  920.97  4979.5  920.97  4980.5  918.97
  5019.5  918.97  5020.5  920.97  5025.5  921.00  5041.0  927.66  5052.6  930.08
  5065.1  929.97  5076.0  931.64  5092.4  937.18  5108.9  941.19  5129.1  947.87
  5156.3  952.75  5171.9  954.39  5207.3  959.94  5219.2  961.00  5224.0  961.83
#Mann=3,-1,0
  4568.6    0.12       0  4979.5    0.04       0  5020.5    0.12       0
Bank Sta=4979.5,5020.5
XS Rating Curve= 0
Exp/Cntr=0.3,0.1

Type RM Length L Ch R = 1,65948,339,339,339
BEGIN DESCRIPTION:
North Hunting Creek 118.5
END DESCRIPTION:
XS GIS Cut Line= 4
      1460841.06       859832.08      1460623.75       859829.83
      1460346.01       859522.97      1460133.24       859366.19
#Sta/Elev= 30
  4386.2  947.83  4510.3  937.14  4561.9  929.90  4631.9  926.49  4672.9  926.96
  4701.1  922.99  4707.1  926.10  4723.2  927.63  4792.9  925.15  4815.3  928.09
  4851.0  929.93  4910.2  928.09  4944.4  929.53  4970.4  920.77  4979.5  920.76
  4980.5  918.76  5019.5  918.76  5020.5  920.76  5029.3  920.76  5029.6  924.88
  5031.5  925.61  5040.9  938.59  5055.5  949.26  5071.0  956.72  5110.8  965.25
  5144.0  969.46  5183.0  972.59  5203.0  976.10  5222.5  976.75  5281.7  982.59
#Mann=3,-1,0
  4386.2    0.12       0  4979.5    0.04       0  5020.5    0.12       0
Bank Sta=4979.5,5020.5
XS Rating Curve= 0
Exp/Cntr=0.3,0.1

Type RM Length L Ch R = 1,65609,481,481,481
BEGIN DESCRIPTION:
North Hunting Creek 118.0
END DESCRIPTION:
XS GIS Cut Line= 4
      1460889.88       859749.45      1460788.45       859621.10
      1460655.93       859385.04      1460591.71       859277.33
#Sta/Elev= 30
  4590.4  948.02  4633.9  946.13  4671.3  943.17  4679.0  943.18  4690.9  942.24
  4730.6  932.93  4765.6  926.19  4791.5  925.22  4816.7  927.00  4826.8  926.63
  4851.2  926.82  4874.0  928.10  4904.7  927.86  4917.6  926.97  4959.7  927.73
  4968.2  926.81  4971.0  922.48  4971.1  920.67  4979.3  920.67  4980.3  918.67
  5019.7  918.67  5020.7  920.67  5031.9  920.67  5040.4  928.24  5043.9  928.56
  5054.7  931.47  5059.7  935.10  5064.6  937.33  5086.4  940.38  5150.1  955.13
#Mann=3,-1,0
  4590.4    0.12       0  4979.3    0.04       0  5020.7    0.12       0
Bank Sta=4979.3,5020.7
XS Rating Curve= 0
Exp/Cntr=0.3,0.1

Type RM Length L Ch R = 1,65128,432,432,432
BEGIN DESCRIPTION:
North Hunting Creek 117.0
END DESCRIPTION:
XS GIS Cut Line= 4
      1461330.98       859542.44      1461204.75       859431.16
      1461090.61       859175.34      1460976.43       859104.47
#Sta/Elev= 30
  4618.7  943.98  4659.9  941.48  4680.5  939.51  4712.9  935.39  4733.4  933.53
  4782.5  930.68  4816.9  926.34  4829.4  925.38  4855.6  925.47  4865.1  924.70
  4944.8  927.61  4959.0  926.66  4966.4  924.14  4967.4  920.65  4979.3  920.65
  4980.3  918.65  5019.7  918.65  5020.7  920.65  5032.7  920.65  5033.3  926.99
  5034.1  928.86  5042.2  927.91  5053.9  927.52  5069.7  930.21  5079.8  932.15
  5098.7  937.08  5113.8  940.00  5156.8  950.83  5183.9  956.76  5201.5  959.52
#Mann=3,-1,0
  4618.7    0.12       0  4979.3    0.04       0  5020.7    0.12       0
Bank Sta=4979.3,5020.7
XS Rating Curve= 0
Exp/Cntr=0.3,0.1

Type RM Length L Ch R = 1,64696,380,380,380
BEGIN DESCRIPTION:
North Hunting Creek 116.5
END DESCRIPTION:
XS GIS Cut Line= 4
      1461497.03       859509.61      1461519.92       859209.01
      1461524.50       859074.74      1461526.02       858995.39
#Sta/Elev= 30
  4591.0  943.92  4649.9  941.37  4674.4  940.91  4727.6  938.98  4750.3  939.23
  4761.8  938.47  4786.9  934.19  4803.6  935.42  4838.7  932.09  4846.6  930.58
  4857.2  929.86  4881.7  927.28  4895.0  925.34  4916.8  923.69  4925.0  924.08
  4941.0  923.93  4955.8  924.36  4974.5  925.37  4975.3  921.21  4975.7  920.64
  4979.3  920.64  4980.3  918.64  5019.7  918.64  5020.7  920.64  5024.3  920.64
  5040.0  926.14  5060.3  942.78  5085.2  952.06  5091.7  953.01  5106.2  956.16
#Mann=3,-1,0
  4591.0    0.12       0  4979.3    0.04       0  5020.7    0.12       0
Bank Sta=4979.3,5020.7
XS Rating Curve= 0
Exp/Cntr=0.3,0.1

Type RM Length L Ch R = 1,64316,297,297,297
BEGIN DESCRIPTION:
North Hunting Creek 116.0
END DESCRIPTION:
XS GIS Cut Line= 4
      1462039.12       859556.92      1462012.20       859314.64
      1461875.54       859043.39      1461616.69       858995.76
#Sta/Elev= 30
  4503.0  943.40  4542.2  938.36  4651.8  932.77  4714.3  932.20  4738.5  930.85
  4807.0  924.36  4825.3  924.59  4856.4  922.56  4902.5  924.76  4942.0  925.16
  4945.6  923.97  4958.7  923.62  4958.8  920.63  4979.3  920.63  4980.3  918.63
  5019.7  918.63  5020.7  920.63  5038.4  920.63  5040.1  925.03  5041.3  925.83
  5050.5  926.46  5109.2  925.61  5193.1  933.62  5240.9  940.91  5264.6  943.54
  5280.9  946.78  5287.5  947.10  5296.7  948.81  5302.0  948.48  5313.7  950.20
#Mann=3,-1,0
  4503.0    0.12       0  4979.3    0.04       0  5020.7    0.12       0
Bank Sta=4979.3,5020.7
XS Rating Curve= 0
Exp/Cntr=0.3,0.1

Type RM Length L Ch R = 1,64019,456,456,456
BEGIN DESCRIPTION:
North Hunting Creek 115.5
END DESCRIPTION:
XS GIS Cut Line= 4
      1462026.51       858714.59      1462023.45       858850.43
      1461786.95       859016.75      1461616.06       858986.24
#Sta/Elev= 30
  4833.2  961.00  4861.9  952.97  4883.8  943.96  4944.5  929.49  4958.7  922.96
  4973.8  920.62  4979.3  920.62  4980.3  918.62  5019.7  918.62  5020.7  920.62
  5037.1  920.62  5037.7  924.90  5048.0  924.83  5051.0  925.92  5062.9  925.40
  5076.7  925.63  5102.0  925.19  5163.9  925.50  5199.0  927.19  5224.7  926.26
  5257.0  928.38  5301.0  933.28  5312.4  932.77  5322.7  934.69  5346.0  937.83
  5373.1  942.27  5385.3  944.04  5388.0  944.67  5409.0  946.70  5431.8  949.96
#Mann=3,-1,0
  4833.2    0.12       0  4979.3    0.04       0  5020.7    0.12       0
Bank Sta=4979.3,5020.7
XS Rating Curve= 0
Exp/Cntr=0.3,0.1

Type RM Length L Ch R = 1,63563,567,567,567
BEGIN DESCRIPTION:
North Hunting Creek 115.0
END DESCRIPTION:
XS GIS Cut Line= 4
      1461703.71       858548.47      1461645.70       858606.48
      1461506.96       858751.43      1461434.48       858840.47
#Sta/Elev= 30
  4882.9  957.41  4892.0  955.31  4935.3  930.04  4941.9  925.96  4956.3  923.45
  4960.0  922.02  4962.2  920.61  4979.3  920.61  4980.3  918.61  5019.7  918.61
  5020.7  920.61  5033.5  920.61  5034.3  923.99  5034.9  924.15  5043.9  924.49
  5047.4  925.47  5056.5  924.62  5064.8  924.61  5073.3  924.89  5081.5  924.93
  5119.5  923.97  5130.6  924.29  5144.2  924.49  5150.3  924.37  5156.4  924.79
  5162.5  925.38  5194.3  934.32  5256.7  953.48  5271.2  957.15  5280.4  959.62
#Mann=3,-1,0
  4882.9    0.12       0  4979.3    0.04       0  5020.7    0.12       0
Bank Sta=4979.3,5020.7
XS Rating Curve= 0
Exp/Cntr=0.3,0.1

Type RM Length L Ch R = 1,62996,262,262,262
BEGIN DESCRIPTION:
North Hunting Creek 114.0
END DESCRIPTION:
XS GIS Cut Line= 4
      1461349.60       858204.77      1461248.13       858217.20
      1461103.19       858326.94      1461024.51       858418.04
#Sta/Elev= 30
  4845.3  941.40  4850.2  940.72  4853.9  940.98  4865.0  939.59  4872.4  937.25
  4881.2  933.80  4893.6  931.86  4915.8  929.19  4931.0  927.71  4937.3  927.48
  4947.5  925.30  4960.6  922.28  4967.9  921.07  4969.0  920.59  4979.3  920.09
  4980.3  918.09  5019.7  918.09  5020.7  920.09  5037.2  920.59  5051.7  923.21
  5087.1  922.28  5130.6  925.38  5134.6  927.20  5164.8  935.53  5192.9  943.04
  5205.1  946.05  5226.7  950.63  5238.3  953.59  5244.8  954.95  5249.7  955.72
#Mann=3,-1,0
  4845.3    0.12       0  4979.3    0.04       0  5020.7    0.12       0
Bank Sta=4979.3,5020.7
XS Rating Curve= 0
Exp/Cntr=0.3,0.1

Type RM Length L Ch R = 1,62734,116,116,116
BEGIN DESCRIPTION:
North Little Hunting Creek 113.5
END DESCRIPTION:
XS GIS Cut Line= 4
      1461357.39       858186.37      1461152.66       858108.23
      1461013.56       857951.94      1461047.95       857847.20
#Sta/Elev= 30
  4682.8  942.14  4689.0  940.07  4706.3  935.73  4731.2  934.38  4766.8  928.74
  4784.2  926.88  4876.2  923.92  4882.4  924.35  4901.9  924.22  4932.0  923.41
  4946.9  921.04  4955.2  916.33  4968.8  915.94  4978.4  914.65  4979.4  912.65
  5020.6  912.65  5021.6  914.65  5025.6  915.04  5043.9  914.65  5059.0  923.52
  5095.0  922.60  5111.2  923.60  5133.6  926.29  5146.7  926.75  5159.4  925.66
  5163.7  927.27  5176.2  933.47  5185.5  937.53  5193.7  942.15  5221.4  949.22
#Mann=3,-1,0
  4682.8    0.12       0  4978.4    0.04       0  5021.6    0.12       0
Bank Sta=4978.4,5021.6
XS Rating Curve= 0
Exp/Cntr=0.5,0.3

Type RM Length L Ch R = 1,62618,35,35,35
BEGIN DESCRIPTION:
Private Rd - US
END DESCRIPTION:
XS GIS Cut Line= 3
      1461361.98       858175.77      1461264.70       858140.59
      1461109.38       857836.17
#Sta/Elev= 30
  4713.6  941.56  4727.0  937.32  4732.3  935.99  4762.5  934.54  4777.3  932.54
  4797.7  929.20  4817.1  927.11  4855.1  925.41  4866.8  925.50  4899.8  922.13
  4905.9  921.14  4927.4  921.47  4934.6  919.95  4951.6  921.88  4964.3  911.11
  4978.4  911.11  4979.4  909.11  5020.6  909.11  5021.6  911.11  5033.4  911.89
  5045.4  920.43  5055.4  926.07  5065.1  928.52  5086.8  927.28  5099.8  932.52
  5106.9  937.98  5127.4  946.71  5142.7  950.22  5148.0  950.80  5158.8  952.81
#Mann=3,-1,0
  4713.6    0.12       0  4978.4    0.04       0  5021.6    0.12       0
Bank Sta=4978.4,5021.6
XS Rating Curve= 0
Exp/Cntr=0.5,0.3

Type RM Length L Ch R =5,62602,,,
BEGIN DESCRIPTION:
Private Rd - TOR
Structure ID: LDS_NLHC_07A
Approximate Survey Structure
END DESCRIPTION:
#Inline Weir SE= 3
  4891.7  922.62  4950.0  922.60  5050.0  922.60
IW Dist,WD,Coef,Skew,MaxSub,Min_El,Is_Ogee,SpillHt,DesHd
14.5,3,3,,0.95,,0,,,1,1

Type RM Length L Ch R = 1,62583,183,183,183
BEGIN DESCRIPTION:
Private Rd - DS
END DESCRIPTION:
XS GIS Cut Line= 3
      1461372.38       858146.80      1461279.19       858103.31
      1461146.65       857827.88
#Sta/Elev= 30
  4751.6  941.52  4779.4  934.65  4804.4  934.42  4827.6  927.12  4851.7  925.63
  4875.1  925.24  4880.2  924.72  4887.8  923.60  4913.5  916.67  4924.4  914.55
  4947.8  912.66  4955.0  911.11  4961.5  910.77  4962.6  909.55  4978.4  908.56
  4979.4  906.06  5020.6  906.06  5021.6  908.56  5026.6  911.11  5034.1  911.24
  5037.6  913.78  5043.2  915.73  5060.8  924.82  5071.0  927.68  5082.3  929.47
  5103.4  928.39  5106.4  930.39  5108.6  931.09  5123.4  945.44  5160.1  952.38
#Mann=3,-1,0
  4751.6    0.12       0  4978.4    0.04       0  5021.6    0.12       0
Bank Sta=4978.4,5021.6
XS Rating Curve= 0
Exp/Cntr=0.5,0.3

Type RM Length L Ch R = 1,62400,241,241,241
BEGIN DESCRIPTION:
North Hunting Creek 113.0
END DESCRIPTION:
XS GIS Cut Line= 4
      1461475.91       858043.27      1461407.57       857939.73
      1461341.31       857861.05      1461217.05       857774.07
#Sta/Elev= 30
  4844.2  943.87  4861.4  939.70  4865.8  937.34  4867.6  936.87  4884.6  929.02
  4889.8  929.27  4907.0  929.10  4913.6  928.73  4932.2  919.54  4936.3  917.10
  4953.3  909.37  4958.1  906.74  4965.9  903.42  4974.1  903.41  4975.3  901.41
  5024.7  901.41  5025.9  903.41  5035.1  903.43  5045.9  906.82  5060.0  907.79
  5073.3  909.18  5151.0  928.48  5157.8  930.50  5178.2  933.49  5197.5  933.06
  5203.0  933.37  5215.6  941.26  5218.7  944.37  5220.2  944.98  5222.8  946.65
#Mann=3,-1,0
  4844.2    0.12       0  4974.1    0.04       0  5025.9    0.12       0
Bank Sta=4974.1,5025.9
XS Rating Curve= 0
Exp/Cntr=0.5,0.3

Type RM Length L Ch R = 1,62159,127,127,127
BEGIN DESCRIPTION:
Buck Shoal Rd - US
END DESCRIPTION:
XS GIS Cut Line= 3
      1461835.75       857990.75      1461638.14       857867.25
      1461438.97       857561.54
#Sta/Elev= 30
  4675.5  944.31  4682.1  944.77  4697.7  942.79  4702.0  943.37  4721.1  941.84
  4732.5  942.26  4772.6  940.09  4829.3  938.36  4864.7  934.81  4886.9  928.03
  4895.2  924.44  4910.8  919.99  4936.9  915.65  4963.1  908.59  4964.6  906.90
  4969.4  901.90  5030.6  901.90  5035.4  906.90  5040.4  912.25  5042.8  912.45
  5049.3  915.01  5054.3  915.49  5079.5  931.24  5092.0  938.17  5096.2  938.87
  5102.3  942.24  5126.7  944.63  5172.9  947.38  5229.9  952.60  5273.4  954.64
#Mann=3,-1,0
  4675.5    0.12       0  4964.6    0.04       0  5035.4    0.12       0
#XS Ineff=2,0
    0.00 4965.00  939.90 5034.00    0.00  939.90
Permanent Ineff=
       F       F
Bank Sta=4964.6,5035.4
XS Rating Curve= 0
Exp/Cntr=0.5,0.3

Type RM Length L Ch R =2,62084,,,
BEGIN DESCRIPTION:
Buck Shoal Rd - TOR
Structure ID: LDS_NLHC_07
Approximate Survey Structure
END DESCRIPTION:
Bridge Culvert--1,0,-1,-1,0
Deck Dist Width WeirC Skew NumUp NumDn MinLoCord MaxHiCord MaxSubmerge Is_Ogee
30,90,3,,4,4,,,,0,1,1,,,
  4746.6  4856.9  5048.1  5147.1
  941.25  939.90  939.90  941.13
  881.90  881.90  881.90  881.90
  4746.6  4856.9  5048.1  5147.1
  941.25  939.90  939.90  941.13
  881.45  881.45  881.45  881.45
Culvert=4,22,50,90,0.013,0.5,1,29,1,902,5000,901.55,5000,Culvert #1,0,30
Culvert Bottom n=0.012
Culvert Bottom Depth=0
Culvert Depth Blocked=0
BC Design=,,0,,0,,,,,,

Type RM Length L Ch R = 1,62032,214,214,214
BEGIN DESCRIPTION:
Buck Shoal Rd - DS
END DESCRIPTION:
XS GIS Cut Line= 3
      1461895.99       857983.05      1461772.46       857890.40
      1461574.85       857513.70
#Sta/Elev= 30
  4720.5  942.42  4783.3  939.81  4796.4  939.65  4799.1  940.18  4813.4  939.38
  4888.1  939.08  4900.2  938.67  4909.3  937.27  4926.9  937.60  4944.9  935.24
  4966.6  934.83  4966.8  934.17  4967.6  905.45  4972.0  901.45  5028.1  901.45
  5032.5  905.45  5039.0  924.78  5041.0  935.24  5073.4  934.27  5092.2  930.87
  5105.4  929.44  5115.4  935.60  5133.5  945.04  5141.2  946.53  5158.0  948.04
  5164.5  952.29  5170.0  953.59  5181.3  958.37  5231.1  968.05  5300.3  977.44
#Mann=3,-1,0
  4720.5    0.12       0  4967.6    0.04       0  5032.5    0.12       0
#XS Ineff=2,0
    0.00 4965.00  932.00 5034.00    0.00  932.00
Permanent Ineff=
       F       F
Bank Sta=4967.6,5032.5
XS Rating Curve= 0
Exp/Cntr=0.5,0.3

Type RM Length L Ch R = 1,61818,662,662,662
BEGIN DESCRIPTION:
North Hunting Creek 112.0
END DESCRIPTION:
XS GIS Cut Line= 4
      1461925.23       857931.44      1461925.23       857825.85
      1461931.45       857736.81      1461937.66       857614.62
#Sta/Elev= 30
  4858.1  930.24  4866.1  928.08  4884.8  923.57  4913.7  917.22  4920.4  915.56
  4924.3  914.53  4934.8  910.42  4943.6  907.66  4949.6  907.12  4961.4  906.26
  4965.9  905.58  4971.7  902.78  4973.7  900.48  4978.4  900.19  4979.4  898.19
  5020.6  898.19  5021.6  900.19  5023.8  900.19  5023.9  900.63  5027.3  900.82
  5054.1  906.45  5071.2  910.50  5083.3  916.46  5100.5  923.31  5120.0  931.33
  5122.4  932.58  5129.0  937.18  5146.8  940.70  5159.1  943.49  5175.3  948.27
#Mann=3,-1,0
  4858.1    0.12       0  4978.4    0.04       0  5021.6    0.12       0
Bank Sta=4978.4,5021.6
XS Rating Curve= 0
Exp/Cntr=0.3,0.1

Type RM Length L Ch R = 1,61156,329,329,329
BEGIN DESCRIPTION:
North Hunting Creek 111.0
END DESCRIPTION:
XS GIS Cut Line= 4
      1462591.99       857900.35      1462602.33       857794.79
      1462422.19       857469.70      1462310.34       857405.49
#Sta/Elev= 30
  4859.2  938.73  4865.5  936.93  4895.0  934.55  4918.4  927.81  4946.5  913.02
  4965.9  898.17  4968.9  897.28  4978.4  897.28  4979.4  895.28  5020.6  895.28
  5021.6  897.28  5032.1  897.44  5032.7  900.91  5058.1  909.99  5067.4  909.06
  5091.8  910.09  5143.3  908.87  5168.4  909.11  5184.3  910.67  5250.8  907.94
  5271.0  909.68  5293.3  909.05  5335.0  911.11  5356.2  915.98  5369.4  923.02
  5376.9  925.05  5390.9  925.40  5409.2  930.14  5423.4  932.27  5465.9  934.70
#Mann=3,-1,0
  4859.2    0.12       0  4978.4    0.04       0  5021.6    0.12       0
Bank Sta=4978.4,5021.6
XS Rating Curve= 0
Exp/Cntr=0.3,0.1

Type RM Length L Ch R = 1,60827,241,241,241
BEGIN DESCRIPTION:
North Little Hunting Creek 110.5
END DESCRIPTION:
XS GIS Cut Line= 4
      1463051.45       857873.87      1462983.13       857776.57
      1462542.08       857281.68      1462355.76       857244.42
#Sta/Elev= 30
  4765.1  955.60  4811.8  947.92  4860.0  935.67  4875.5  932.36  4883.9  931.55
  4899.5  927.40  4923.3  918.42  4927.8  915.69  4950.5  908.98  4967.8  900.38
  4970.3  896.54  4978.4  896.54  4979.4  894.54  5020.6  894.54  5021.6  896.54
  5034.6  896.67  5036.0  898.21  5073.5  908.59  5111.9  907.39  5149.3  908.38
  5172.0  910.36  5308.1  910.45  5532.9  907.65  5553.3  910.28  5575.7  915.97
  5588.2  920.38  5595.7  921.13  5650.1  931.84  5718.9  941.03  5736.9  941.20
#Mann=3,-1,0
  4765.1    0.12       0  4978.4    0.04       0  5021.6    0.12       0
Bank Sta=4978.4,5021.6
XS Rating Curve= 0
Exp/Cntr=0.3,0.1

Type RM Length L Ch R = 1,60586,489,489,489
BEGIN DESCRIPTION:
North Hunting Creek 110.0
END DESCRIPTION:
XS GIS Cut Line= 4
      1463206.94       857699.50      1463138.63       857602.22
      1462697.58       857107.33      1462511.24       857070.06
#Sta/Elev= 30
  4855.7  941.25  4899.7  932.64  4907.6  929.82  4936.6  915.09  4949.3  906.97
  4954.9  905.05  4958.2  900.57  4963.8  896.03  4978.4  896.01  4979.4  894.01
  5020.6  894.01  5021.6  896.01  5035.9  896.01  5039.5  898.15  5067.2  907.69
  5101.2  908.87  5108.8  906.04  5142.2  904.25  5148.7  904.95  5160.9  910.45
  5167.8  910.61  5199.0  908.72  5311.2  909.91  5367.1  908.65  5484.5  908.35
  5546.0  906.38  5625.1  907.56  5705.4  913.39  5796.1  924.76  5827.5  927.56
#Mann=3,-1,0
  4855.7    0.12       0  4978.4    0.04       0  5021.6    0.12       0
#XS Ineff=2,0
       0                 5101.20    0.00  908.87
Permanent Ineff=
       F       F
Bank Sta=4978.4,5021.6
XS Rating Curve= 0
Exp/Cntr=0.3,0.1

Type RM Length L Ch R = 1,60097,371,371,371
BEGIN DESCRIPTION:
North Hunting Creek 109.0
END DESCRIPTION:
XS GIS Cut Line= 4
      1463730.15       857416.01      1463555.03       857321.56
      1463330.69       857132.64      1463210.64       856768.58
#Sta/Elev= 30
  4716.3  952.10  4780.2  947.40  4801.8  943.88  4845.6  931.39  4859.8  925.06
  4880.4  921.63  4905.2  912.03  4936.2  903.61  4960.7  902.03  4970.1  893.75
  4978.4  893.75  4979.4  891.75  5020.6  891.75  5021.6  893.75  5032.4  894.03
  5043.7  904.52  5065.8  907.22  5088.3  906.91  5118.2  900.62  5151.5  900.46
  5162.9  897.90  5176.7  898.28  5179.3  895.18  5183.9  895.11  5190.8  896.47
  5198.7  901.30  5252.4  914.69  5302.4  919.14  5465.8  914.20  5591.9  921.57
#Mann=3,-1,0
  4716.3    0.12       0  4978.4    0.04       0  5021.6    0.12       0
#XS Ineff=2,0
       0                 5065.80    0.00  907.22
Permanent Ineff=
       F       F
Bank Sta=4978.4,5021.6
XS Rating Curve= 0
Exp/Cntr=0.3,0.1

Type RM Length L Ch R = 1,59726,495,495,495
BEGIN DESCRIPTION:
North Hunting Creek 108.5
END DESCRIPTION:
XS GIS Cut Line= 4
      1464054.73       857171.28      1463883.24       857062.97
      1463341.82       856823.84      1463219.97       856756.15
#Sta/Elev= 30
  4638.8  950.10  4667.3  946.81  4696.0  941.67  4743.8  935.05  4763.9  931.22
  4810.6  919.20  4822.5  917.20  4860.3  915.46  4882.8  913.09  4901.9  913.84
  4924.3  912.64  4935.1  907.86  4950.5  902.98  4956.6  897.36  4956.8  892.91
  4978.2  892.90  4979.2  890.90  5020.8  890.90  5021.8  892.90  5038.4  892.90
  5039.7  897.57  5048.4  904.04  5052.4  904.48  5157.1  905.60  5213.7  902.79
  5247.6  902.88  5314.3  908.63  5417.7  909.42  5460.0  911.51  5572.9  921.91
#Mann=3,-1,0
  4638.8    0.12       0  4978.2    0.04       0  5021.8    0.12       0
#XS Ineff=2,0
       0                 5082.60    0.00  905.43
Permanent Ineff=
       F       F
Bank Sta=4978.2,5021.8
XS Rating Curve= 0
Exp/Cntr=0.3,0.1

Type RM Length L Ch R = 1,59231,199,199,199
BEGIN DESCRIPTION:
North Hunting Creek 108.0
END DESCRIPTION:
XS GIS Cut Line= 4
      1464057.05       856778.42      1463972.42       856550.13
      1463433.21       856469.45      1463333.29       856378.48
#Sta/Elev= 30
  4660.7  940.38  4684.3  938.70  4740.7  929.69  4753.5  929.02  4788.8  924.31
  4813.6  920.69  4831.7  916.05  4850.1  913.43  4904.7  909.91  4957.4  909.29
  4971.5  898.22  4973.2  892.84  4978.0  892.84  4979.0  890.84  5021.0  890.84
  5022.0  892.84  5030.7  892.84  5040.9  898.25  5066.3  904.26  5100.2  902.59
  5157.1  901.82  5195.0  902.09  5264.9  904.87  5352.6  903.90  5414.2  905.83
  5437.7  907.61  5496.7  914.77  5520.4  920.05  5542.9  923.53  5584.5  926.30
#Mann=3,-1,0
  4660.7    0.12       0  4978.0    0.04       0  5022.0    0.12       0
#XS Ineff=2,0
       0                 5066.30    0.00  904.86
Permanent Ineff=
       F       F
Bank Sta=4978,5022
XS Rating Curve= 0
Exp/Cntr=0.5,0.3

Type RM Length L Ch R = 1,59032,277,277,277
BEGIN DESCRIPTION:
Hwy 77 - US
END DESCRIPTION:
XS GIS Cut Line= 4
      1464062.58       856781.88      1463977.39       856541.11
      1463836.61       856229.92      1463693.97       855961.30
#Sta/Elev= 30
  4523.0  940.02  4558.2  937.70  4606.5  930.80  4620.0  930.10  4647.1  926.63
  4683.9  921.43  4705.6  915.94  4720.7  913.21  4730.8  913.67  4743.9  911.05
  4753.8  912.03  4773.9  910.63  4784.6  910.91  4792.2  909.61  4817.3  909.87
  4837.6  907.30  4856.8  908.30  4870.7  907.85  4877.2  906.56  4888.2  906.49
  4920.5  903.78  4937.1  903.68  4960.4  901.20  4970.0  890.70  5030.0  890.70
  5039.6  901.20  5088.8  902.62  5215.4  914.41  5250.5  916.41  5424.1  922.56
#Mann=3,-1,0
  4523.0    0.09       0  4960.4    0.04       0  5039.6    0.09       0
#XS Ineff=2,0
    0.00 4883.00  933.26 5117.00    0.00  933.11
Permanent Ineff=
       F       F
Bank Sta=4960.4,5039.6
XS Rating Curve= 0
Exp/Cntr=0.5,0.3

Type RM Length L Ch R =3,58903,,,
BEGIN DESCRIPTION:
Hwy 77 - TOR
Structure ID: LDS_NLHC_05
Approximate Survey Structure
END DESCRIPTION:
Bridge Culvert--1,0,-1,-1,0
Deck Dist Width WeirC Skew NumUp NumDn MinLoCord MaxHiCord MaxSubmerge Is_Ogee
106.5,90,3,,6,6,,,0.95,0,1.0,1,,,
  4428.2  4892.5  4892.5  5107.5  5107.5  5423.8
  939.09  933.10  933.10  933.10  933.10  932.27
  870.70  870.70  928.60  928.60  870.70  870.70
  4428.2  4892.5  4892.5  5107.5  5107.5  5423.8
  939.09  933.10  933.10  933.10  933.10  932.27
  870.70  870.70  928.60  928.60  870.70  870.70
Pier Skew, UpSta & Num, DnSta & Num=,4946.3,2,4946.3,2,0,0,0,0,0
     2.7     2.7
  897.48  928.60
     2.7     2.7
  903.02  928.60
Pier Skew, UpSta & Num, DnSta & Num=,5053.8,2,5053.8,2,0,0,0,0,0
     2.7     2.7
  901.22  928.60
     2.7     2.7
  899.92  928.60
Abutment Skew #Up #Dn=,2,2
  4892.5  4927.5
  928.60  903.69
  4892.5  4927.5
  928.60  903.96
Abutment Skew #Up #Dn=,2,2
  5072.5  5107.5
  901.71  928.60
  5072.5  5107.5
  901.26  928.60
BR Coef=1,1,0,1.25,0,,,0.8,0,2,0,
WSPro=,,,, 1 ,,,, 0 ,,,, 0 ,,,,-1 ,-1 ,-1 , 0 , 0 , 0 , 0 , 0
BC Design=,,0,,0,,,,,,

Type RM Length L Ch R = 1,58755,190,190,190
BEGIN DESCRIPTION:
Hwy 77 - DS
END DESCRIPTION:
XS GIS Cut Line= 3
      1464531.18       856626.28      1464205.22       856409.59
      1463973.68       855857.60
#Sta/Elev= 30
  4401.9  954.06  4520.7  949.08  4652.3  942.17  4724.3  939.62  4787.9  935.91
  4805.7  933.73  4827.9  929.12  4835.8  926.39  4850.5  922.80  4879.5  912.12
  4885.0  912.70  4907.5  906.81  4932.7  902.93  4956.3  902.78  4960.4  899.45
  4970.0  890.45  5030.0  890.45  5039.6  899.45  5042.2  900.06  5060.1  900.01
  5094.4  903.21  5114.7  906.86  5123.6  907.25  5154.4  912.47  5177.1  914.32
  5216.2  919.62  5258.3  923.56  5301.3  929.13  5322.3  930.47  5391.9  938.44
#Mann=3,-1,0
  4401.9    0.09       0  4960.4    0.04       0  5039.6    0.09       0
#XS Ineff=2,0
    0.00 4883.00  929.40 5117.00    0.00  929.40
Permanent Ineff=
       F       F
Bank Sta=4960.4,5039.6
XS Rating Curve= 0
Exp/Cntr=0.5,0.3

Type RM Length L Ch R = 1,58565,225,225,225
BEGIN DESCRIPTION:
North Hunting Creek 107.0
END DESCRIPTION:
XS GIS Cut Line= 4
      1464409.99       856276.98      1464349.96       856183.82
      1464194.66       856057.51      1464122.21       855925.03
#Sta/Elev= 30
  4815.1  926.87  4840.9  923.20  4854.2  921.54  4867.5  920.30  4878.2  916.75
  4884.9  914.79  4916.0  907.92  4918.7  907.51  4925.9  905.67  4956.8  898.49
  4972.7  892.11  4978.0  892.11  4979.0  890.11  5021.0  890.11  5022.0  892.11
  5032.3  892.11  5046.4  899.20  5061.1  901.66  5076.5  901.65  5100.1  902.50
  5112.4  903.14  5142.1  905.67  5160.6  907.61  5172.2  909.40  5185.6  911.04
  5195.9  911.72  5199.8  912.36  5236.0  916.74  5258.3  919.00  5277.1  921.56
#Mann=3,-1,0
  4815.1    0.09       0  4978.0    0.04       0  5022.0    0.12       0
Bank Sta=4978,5022
XS Rating Curve= 0
Exp/Cntr=0.3,0.1

Type RM Length L Ch R = 1,58340,330,330,330
BEGIN DESCRIPTION:
North Little Hunting Creek 106.5
END DESCRIPTION:
XS GIS Cut Line= 4
      1464562.88       855953.81      1464377.71       855934.19
      1464310.25       855901.08      1464203.58       855818.92
#Sta/Elev= 30
  4786.2  929.88  4803.7  928.91  4821.0  928.26  4853.5  923.51  4878.2  919.51
  4882.4  918.44  4889.3  917.21  4903.4  915.22  4915.7  910.70  4919.4  909.11
  4931.7  904.84  4942.9  900.49  4947.5  900.06  4960.1  896.70  4972.4  892.31
  4978.0  889.96  4979.0  887.96  5021.0  887.96  5022.0  889.96  5027.5  890.37
  5029.7  891.62  5038.9  891.06  5047.6  891.51  5086.5  899.63  5098.8  902.49
  5121.3  908.60  5150.0  915.31  5175.7  920.62  5179.0  921.05  5182.2  921.87
#Mann=3,-1,0
  4786.2    0.09       0  4978.0    0.04       0  5022.0    0.12       0
Bank Sta=4978,5022
XS Rating Curve= 0
Exp/Cntr=0.3,0.1
