HEC-RAS study North Little Hunting Creek.prj: North Little Hunting Creek Limited Detail Study

--- North Little Hunting Creek.g01 (geometry) --- (continued)

Type RM Length L Ch R = 1,58010,578,578,578
BEGIN DESCRIPTION:
North Hunting Creek 106.0
END DESCRIPTION:
XS GIS Cut Line= 4
      1464606.70       855728.26      1464511.47       855637.17
      1464453.49       855601.97      1464354.12       855537.79
#Sta/Elev= 30
  4835.1  919.38  4841.1  918.21  4849.9  917.01  4858.4  915.31  4870.3  912.53
  4896.5  905.70  4908.0  901.20  4911.7  900.31  4917.3  898.37  4919.7  897.76
  4929.7  896.61  4945.3  896.17  4966.8  890.95  4974.7  888.41  4978.0  888.41
  4979.0  886.41  5021.0  886.41  5022.0  888.41  5023.2  888.50  5029.2  890.42
  5058.4  901.29  5060.9  902.06  5070.9  904.32  5081.3  907.70  5082.8  908.00
  5098.9  913.68  5101.3  914.76  5118.1  917.81  5141.7  920.31  5153.0  922.14
#Mann=3,-1,0
  4835.1    0.09       0  4978.0    0.04       0  5022.0    0.12       0
Bank Sta=4978,5022
XS Rating Curve= 0
Exp/Cntr=0.3,0.1

Type RM Length L Ch R = 1,57432,364,364,364
BEGIN DESCRIPTION:
North Hunting Creek 105.0
END DESCRIPTION:
XS GIS Cut Line= 4
      1465122.35       855436.35      1465004.29       855343.14
      1464913.18       855249.96      1464830.38       855163.02
#Sta/Elev= 30
  4753.8  915.96  4797.9  913.05  4836.4  909.86  4864.1  906.21  4883.3  902.40
  4893.5  900.89  4901.8  899.96  4909.0  899.54  4916.7  898.90  4929.2  897.09
  4934.2  897.01  4950.3  896.02  4957.2  893.57  4960.4  892.79  4970.9  889.10
  4971.4  887.85  4971.7  885.44  4977.9  884.36  4978.9  882.36  5021.1  882.36
  5022.1  884.36  5030.4  885.44  5031.4  884.36  5036.0  886.08  5039.8  888.58
  5050.7  894.14  5059.1  897.63  5078.3  899.39  5125.8  911.24  5154.6  916.88
#Mann=4,-1,0
  4753.8    0.06       0  4909.0    0.12       0  4977.9    0.04       0
  5022.1    0.12       0
Bank Sta=4977.9,5022.1
XS Rating Curve= 0
Exp/Cntr=0.3,0.1

Type RM Length L Ch R = 1,57068,348,348,348
BEGIN DESCRIPTION:
North Hunting Creek 104.5
END DESCRIPTION:
XS GIS Cut Line= 4
      1465370.59       855208.21      1465284.89       855103.47
      1465166.80       854991.09      1464964.87       854935.85
#Sta/Elev= 30
  4750.2  917.91  4783.9  914.97  4806.1  911.83  4850.4  903.53  4861.2  901.94
  4880.8  896.22  4917.4  893.79  4925.2  893.75  4952.5  891.53  4961.1  889.40
  4968.2  883.34  4977.9  882.66  4978.9  880.66  5021.1  880.66  5022.1  882.66
  5025.0  882.67  5025.5  890.41  5030.3  895.20  5036.4  897.18  5056.7  896.46
  5065.8  898.40  5078.1  899.20  5087.4  901.12  5099.6  902.05  5152.5  910.67
  5189.7  915.20  5198.6  917.04  5214.7  919.38  5245.0  922.65  5257.9  925.48
#Mann=3,-1,0
  4750.2    0.12       0  4977.9    0.04       0  5022.1    0.12       0
Bank Sta=4977.9,5022.1
XS Rating Curve= 0
Exp/Cntr=0.3,0.1

Type RM Length L Ch R = 1,56720,634,634,634
BEGIN DESCRIPTION:
North Hunting Creek 104.0
END DESCRIPTION:
XS GIS Cut Line= 4
      1465662.74       855090.51      1465563.36       854947.65
      1465486.75       854829.62      1465418.43       854738.53
#Sta/Elev= 30
  4704.3  916.31  4726.5  914.32  4750.5  912.56  4796.1  908.68  4817.0  907.25
  4839.1  905.35  4859.4  901.19  4867.6  900.47  4885.9  897.89  4899.4  896.55
  4919.8  895.37  4950.9  894.88  4960.9  889.09  4974.4  882.64  4977.9  882.64
  4978.9  880.64  5021.1  880.64  5022.1  882.64  5029.4  892.03  5032.7  894.97
  5036.3  895.62  5053.9  900.76  5063.8  903.10  5069.8  904.22  5095.9  910.51
  5103.6  911.40  5105.8  911.98  5118.7  913.99  5122.2  913.68  5132.9  914.26
#Mann=3,-1,0
  4704.3    0.12       0  4977.9    0.04       0  5022.1    0.12       0
Bank Sta=4977.9,5022.1
XS Rating Curve= 0
Exp/Cntr=0.3,0.1

Type RM Length L Ch R = 1,56086,318,318,318
BEGIN DESCRIPTION:
North Hunting Creek 103.0
END DESCRIPTION:
XS GIS Cut Line= 4
      1466199.03       854643.23      1466085.16       854500.39
      1465888.45       854384.43      1465741.40       854367.86
#Sta/Elev= 30
  4643.3  904.17  4669.0  903.89  4717.8  902.56  4765.6  900.00  4817.6  896.12
  4838.3  894.99  4897.0  893.72  4920.4  893.84  4938.6  893.40  4940.0  892.96
  4953.0  892.51  4956.1  891.83  4959.8  892.70  4969.5  882.60  4977.9  882.60
  4978.9  880.60  5021.1  880.60  5022.1  882.60  5029.1  882.60  5030.7  885.40
  5037.9  891.20  5042.2  895.96  5076.5  896.82  5088.4  897.91  5101.7  899.99
  5111.7  901.08  5154.7  909.35  5187.3  913.30  5196.9  914.09  5202.3  914.06
#Mann=4,-1,0
  4643.3    0.06       0  4897.0    0.12       0  4977.9    0.04       0
  5022.1    0.12       0
Bank Sta=4977.9,5022.1
XS Rating Curve= 0
Exp/Cntr=0.3,0.1

Type RM Length L Ch R = 1,55768,510,510,510
BEGIN DESCRIPTION:
North Hunting Creek 102.5
END DESCRIPTION:
XS GIS Cut Line= 4
      1466232.05       854636.50      1466262.85       854379.06
      1466141.85       854148.05      1466100.04       854000.62
#Sta/Elev= 30
  4532.9  904.01  4641.5  903.32  4696.5  901.67  4746.3  898.63  4799.3  893.47
  4821.7  892.82  4842.8  892.61  4892.0  894.37  4919.1  895.49  4925.9  895.10
  4945.5  892.09  4951.4  889.61  4962.1  882.65  4977.9  882.58  4978.9  880.58
  5021.1  880.58  5022.1  882.58  5029.8  882.58  5030.0  884.89  5031.2  890.47
  5038.3  892.77  5048.4  893.88  5072.9  906.93  5098.1  914.09  5112.8  916.09
  5130.3  917.26  5164.7  921.05  5171.3  922.83  5178.7  922.04  5206.2  924.84
#Mann=4,-1,0
  4532.9    0.06       0  4892.0    0.12       0  4977.9    0.04       0
  5022.1    0.12       0
#XS Ineff=2,0
    0.00 4917.10  895.39               0
Permanent Ineff=
       F       F
Bank Sta=4977.9,5022.1
XS Rating Curve= 0
Exp/Cntr=0.3,0.1

Type RM Length L Ch R = 1,55258,582,582,582
BEGIN DESCRIPTION:
North Hunting Creek 102.0
END DESCRIPTION:
XS GIS Cut Line= 4
      1466269.47       854651.52      1466389.55       854413.42
      1466491.01       854295.39      1466559.32       854243.65
#Sta/Elev= 30
  4650.8  903.86  4749.3  902.48  4808.2  900.90  4896.9  896.09  4905.0  895.25
  4934.0  892.59  4948.8  892.09  4955.6  892.07  4966.5  891.53  4968.5  889.82
  4977.9  879.28  4978.9  877.28  5021.1  877.28  5022.1  879.28  5025.2  879.29
  5027.0  879.80  5029.6  879.31  5034.1  879.75  5039.6  883.23  5059.1  889.58
  5063.8  890.00  5079.9  890.52  5084.2  893.15  5102.8  902.10  5116.0  912.29
  5130.6  925.80  5135.6  929.36  5144.9  940.44  5148.0  943.79  5158.8  952.20
#Mann=4,-1,0
  4650.8    0.06       0  4905.0    0.12       0  4977.9    0.04       0
  5022.1    0.12       0
Bank Sta=4977.9,5022.1
XS Rating Curve= 0
Exp/Cntr=0.3,0.1

Type RM Length L Ch R = 1,54676,606,606,606
BEGIN DESCRIPTION:
North Hunting Creek 101.0
END DESCRIPTION:
XS GIS Cut Line= 4
      1466464.09       854871.03      1466590.40       854871.03
      1466733.28       854868.96      1466832.67       854829.62
#Sta/Elev= 30
  4793.9  910.82  4816.1  908.93  4851.4  904.60  4866.0  903.06  4899.6  900.37
  4914.9  897.69  4924.7  896.31  4942.9  892.06  4957.2  890.92  4960.9  891.11
  4969.2  880.70  4970.1  879.84  4970.5  878.80  4977.9  878.80  4978.9  876.80
  5021.1  876.80  5022.1  878.80  5029.3  878.80  5031.8  886.32  5032.2  886.82
  5046.1  889.53  5047.6  890.25  5054.4  892.46  5061.6  895.39  5077.1  899.27
  5098.2  915.60  5126.3  927.85  5139.8  932.80  5160.6  937.74  5170.0  939.45
#Mann=3,-1,0
  4793.9    0.12       0  4977.9    0.04       0  5022.1    0.12       0
Bank Sta=4977.9,5022.1
XS Rating Curve= 0
Exp/Cntr=0.3,0.1

Type RM Length L Ch R = 1,54070,475,475,475
BEGIN DESCRIPTION:
North Hunting Creek 100.0
END DESCRIPTION:
XS GIS Cut Line= 4
      1466391.62       855463.24      1466497.22       855467.38
      1466673.23       855473.59      1466782.97       855411.47
#Sta/Elev= 30
  4747.2  926.06  4753.2  923.94  4771.7  918.34  4790.2  913.32  4809.5  907.43
  4822.1  904.22  4843.3  897.08  4859.0  896.27  4860.2  896.09  4870.6  892.77
  4878.7  891.05  4883.0  890.64  4897.3  888.43  4911.1  887.81  4920.7  884.48
  4928.1  883.24  4931.3  880.87  4961.4  884.99  4972.9  885.79  4977.9  878.33
  4978.9  876.33  5021.1  876.33  5022.1  878.33  5029.0  878.33  5058.1  902.31
  5063.9  906.80  5082.0  908.38  5087.2  909.41  5131.1  915.43  5155.1  918.08
#Mann=3,-1,0
  4747.2    0.12       0  4977.9    0.04       0  5022.1    0.12       0
Bank Sta=4977.9,5022.1
XS Rating Curve= 0
Exp/Cntr=0.3,0.1

Type RM Length L Ch R = 1,53595,323,323,323
BEGIN DESCRIPTION:
North Hunting Creek 99.0
END DESCRIPTION:
XS GIS Cut Line= 4
      1466913.42       855858.74      1466907.21       855773.84
      1466898.93       855676.52      1466884.43       855521.19
#Sta/Elev= 30
  4894.4  922.47  4907.3  918.61  4916.2  915.54  4927.5  906.59  4950.6  892.18
  4965.6  885.17  4975.2  876.84  4977.9  876.68  4978.9  874.68  5021.1  874.68
  5022.1  876.68  5026.8  876.68  5028.7  878.52  5032.2  880.02  5042.0  885.01
  5044.4  886.69  5066.0  888.28  5071.6  890.43  5079.0  891.87  5082.3  891.91
  5098.4  890.64  5109.3  891.30  5127.2  891.79  5142.4  894.35  5172.6  900.58
  5178.5  901.15  5188.0  903.30  5204.3  905.50  5219.2  908.95  5233.2  910.17
#Mann=3,-1,0
  4894.4    0.12       0  4977.9    0.04       0  5022.1    0.12       0
Bank Sta=4977.9,5022.1
XS Rating Curve= 0
Exp/Cntr=0.3,0.1

Type RM Length L Ch R = 1,53272,271,271,271
BEGIN DESCRIPTION:
North Little Hunting Creek 98.5
END DESCRIPTION:
XS GIS Cut Line= 3
      1467232.95       855625.32      1467148.24       855554.73
      1467005.93       855434.76
#Sta/Elev= 28
  4871.0  939.75  4877.5  937.52  4883.2  936.05  4887.4  933.82  4894.3  930.78
  4906.7  923.65  4910.5  921.77  4922.4  915.43  4929.5  912.21  4937.6  906.66
  4943.8  902.17  4953.8  896.44  4960.3  892.19  4966.2  888.65  4968.8  886.16
  4976.6  875.84  4977.6  873.84  5022.4  873.84  5023.4  875.84  5026.4  875.86
  5030.1  877.67  5033.9  884.21  5092.4  890.44  5105.5  890.08  5125.5  895.63
  5139.5  899.40  5161.4  904.27  5167.4  905.68
#Mann=3,-1,0
  4871.0    0.12       0  4976.6    0.04       0  5023.4    0.12       0
Bank Sta=4976.6,5023.4
XS Rating Curve= 0
Exp/Cntr=0.3,0.1

Type RM Length L Ch R = 1,53001,641,641,641
BEGIN DESCRIPTION:
North Hunting Creek 98.0
END DESCRIPTION:
XS GIS Cut Line= 4
      1467412.41       855421.80      1467339.98       855361.78
      1467228.16       855283.09      1467135.02       855235.49
#Sta/Elev= 30
  4799.8  923.26  4809.4  919.56  4825.5  912.50  4835.7  907.06  4852.4  900.41
  4856.6  898.29  4883.5  887.10  4888.5  885.44  4905.6  883.27  4912.9  884.05
  4928.9  883.68  4933.2  884.65  4939.1  883.99  4948.8  884.20  4959.4  880.09
  4969.6  876.75  4972.1  875.31  4976.6  875.28  4977.6  873.28  5022.4  873.28
  5023.4  875.28  5035.8  875.32  5038.8  877.00  5042.1  877.94  5070.9  889.80
  5081.0  892.57  5095.4  898.54  5109.1  903.11  5118.4  904.37  5135.2  907.88
#Mann=3,-1,0
  4799.8    0.12       0  4976.6    0.04       0  5023.4    0.12       0
Bank Sta=4976.6,5023.4
XS Rating Curve= 0
Exp/Cntr=0.3,0.1

Type RM Length L Ch R = 1,52360,601,601,601
BEGIN DESCRIPTION:
North Hunting Creek 97.0
END DESCRIPTION:
XS GIS Cut Line= 4
      1467834.81       854916.57      1467756.18       854887.60
      1467665.07       854821.34      1467598.81       854765.43
#Sta/Elev= 28
  4840.5  910.34  4842.3  909.85  4847.1  908.24  4862.3  902.41  4878.2  896.67
  4882.2  895.71  4885.2  894.43  4892.9  891.96  4899.4  889.53  4920.7  884.08
  4927.4  882.48  4940.9  881.01  4946.0  880.29  4948.1  879.60  4963.8  871.92
  4976.6  872.92  4977.6  870.92  5022.4  870.92  5023.4  872.92  5026.8  872.64
  5068.2  884.12  5079.9  888.76  5083.0  890.42  5095.1  897.57  5103.0  902.09
  5110.4  904.03  5121.2  907.22  5123.7  907.51
#Mann=3,-1,0
  4840.5    0.12       0  4976.6    0.04       0  5023.4    0.12       0
Bank Sta=4976.6,5023.4
XS Rating Curve= 0
Exp/Cntr=0.3,0.1

Type RM Length L Ch R = 1,51759,607,607,607
BEGIN DESCRIPTION:
North Hunting Creek 96.0
END DESCRIPTION:
XS GIS Cut Line= 4
      1468168.22       854450.68      1468108.19       854403.07
      1468012.94       854338.88      1467932.22       854285.06
#Sta/Elev= 30
  4904.0  909.05  4919.0  901.25  4920.7  900.05  4932.7  893.21  4949.6  884.30
  4953.8  882.28  4964.9  873.78  4968.4  871.90  4968.5  870.97  4976.6  872.10
  4977.6  870.10  5022.4  870.10  5023.4  872.10  5039.2  870.97  5041.8  870.97
  5050.1  880.59  5063.4  880.09  5070.5  880.65  5073.4  880.00  5076.0  879.81
  5093.7  879.31  5110.0  881.87  5116.7  883.56  5132.9  886.46  5138.8  888.96
  5150.8  892.16  5160.3  895.55  5171.5  899.00  5178.0  901.67  5192.5  908.60
#Mann=3,-1,0
  4904.0    0.12       0  4976.6    0.04       0  5023.4    0.12       0
Bank Sta=4976.6,5023.4
XS Rating Curve= 0
Exp/Cntr=0.3,0.1

Type RM Length L Ch R = 1,51152,234,234,234
BEGIN DESCRIPTION:
North Hunting Creek 95.0
END DESCRIPTION:
XS GIS Cut Line= 4
      1468491.29       853885.41      1468435.35       853877.12
      1468255.20       853866.77      1468149.61       853937.16
#Sta/Elev= 30
  4907.3  905.64  4911.9  902.97  4914.3  901.96  4917.3  899.61  4935.9  887.77
  4946.4  882.23  4957.0  876.26  4967.5  870.81  4976.6  871.97  4977.6  869.97
  5022.4  869.97  5023.4  871.97  5029.2  870.81  5037.2  875.02  5042.6  877.22
  5048.1  876.84  5059.4  877.70  5067.5  877.21  5080.7  878.22  5090.6  880.56
  5100.0  884.07  5113.9  888.77  5132.3  893.31  5167.9  896.07  5179.6  895.98
  5190.1  897.09  5216.2  899.98  5239.7  903.98  5262.5  907.13  5271.2  908.08
#Mann=3,-1,0
  4907.3    0.12       0  4976.6    0.04       0  5023.4    0.12       0
Bank Sta=4976.6,5023.4
XS Rating Curve= 0
Exp/Cntr=0.3,0.1

Type RM Length L Ch R = 1,50918,212,212,212
BEGIN DESCRIPTION:
North Little Hunting Creek 94.5
END DESCRIPTION:
XS GIS Cut Line= 4
      1468514.57       853600.19      1468437.27       853627.16
      1468318.20       853665.92      1468153.91       853637.05
#Sta/Elev= 30
  4862.8  934.55  4866.5  933.26  4884.7  923.29  4890.3  920.71  4893.6  918.21
  4902.3  913.36  4918.7  901.14  4926.8  896.60  4940.3  881.36  4959.9  873.04
  4966.8  870.69  4970.4  870.09  4971.6  868.09  5028.4  868.09  5029.6  870.09
  5047.0  876.57  5068.7  878.29  5094.3  877.40  5125.9  879.39  5144.4  880.20
  5147.7  880.69  5166.2  882.16  5170.5  882.24  5187.9  883.57  5193.6  883.60
  5196.2  883.98  5211.1  885.25  5215.9  885.04  5233.4  887.63  5236.7  887.89
#Mann=3,-1,0
  4862.8    0.12       0  4970.4    0.04       0  5029.6    0.12       0
Bank Sta=4970.4,5029.6
XS Rating Curve= 0
Exp/Cntr=0.3,0.1

Type RM Length L Ch R = 1,50706,181,181,181
BEGIN DESCRIPTION:
North Hunting Creek 94.0
END DESCRIPTION:
XS GIS Cut Line= 4
      1468381.48       853417.45      1468302.83       853452.64
      1468207.58       853487.84      1468033.62       853452.63
#Sta/Elev= 30
  4895.2  916.26  4899.0  915.72  4901.3  915.17  4914.3  911.59  4924.5  907.62
  4934.8  902.09  4974.4  870.92  4975.3  869.49  4976.3  867.49  5023.7  867.49
  5024.7  869.49  5028.6  870.11  5030.4  871.26  5056.4  874.39  5086.3  876.15
  5107.5  878.00  5110.5  878.41  5113.1  879.19  5123.2  880.66  5130.2  881.59
  5137.1  882.10  5147.5  883.49  5162.6  886.05  5168.6  886.44  5179.5  888.52
  5188.6  890.02  5203.1  892.96  5209.2  894.62  5238.0  901.21  5260.4  904.76
#Mann=3,-1,0
  4895.2    0.12       0  4975.3    0.04       0  5024.7    0.12       0
Bank Sta=4975.3,5024.7
XS Rating Curve= 0
Exp/Cntr=0.3,0.1

Type RM Length L Ch R = 1,50525,323,323,323
BEGIN DESCRIPTION:
North Little Hunting Creek 93.5
END DESCRIPTION:
XS GIS Cut Line= 4
      1468379.81       853377.35      1468284.51       853267.00
      1468118.94       853332.22      1468028.58       853362.34
#Sta/Elev= 30
  4754.9  911.66  4768.5  908.60  4792.8  905.30  4807.9  902.95  4821.1  899.89
  4831.6  899.06  4837.4  897.45  4851.7  893.98  4875.3  886.24  4895.2  880.89
  4900.7  879.95  4906.8  879.41  4914.9  879.39  4946.6  877.33  4960.5  873.90
  4975.3  867.78  4976.3  865.78  5023.7  865.78  5024.7  867.78  5026.5  867.16
  5027.2  871.00  5028.3  874.81  5067.1  874.56  5077.7  875.88  5086.5  877.60
  5114.8  883.68  5145.3  893.36  5154.8  896.82  5169.7  902.68  5173.9  903.93
#Mann=3,-1,0
  4754.9    0.12       0  4975.3    0.04       0  5024.7    0.12       0
Bank Sta=4975.3,5024.7
XS Rating Curve= 0
Exp/Cntr=0.3,0.1

Type RM Length L Ch R = 1,50202,598,598,598
BEGIN DESCRIPTION:
North Hunting Creek 93.0
END DESCRIPTION:
XS GIS Cut Line= 4
      1468358.76       852914.26      1468265.55       852951.54
      1467948.75       853042.65      1467884.59       853115.09
#Sta/Elev= 30
  4693.7  898.59  4704.1  894.30  4744.0  882.78  4752.1  880.88  4762.3  881.09
  4796.0  880.14  4836.3  877.84  4866.9  877.46  4879.1  876.32  4892.4  876.91
  4930.7  873.93  4950.1  873.96  4964.6  867.92  4975.3  865.33  4976.3  863.33
  5023.7  863.33  5024.7  865.33  5030.7  865.34  5031.5  871.16  5040.8  873.51
  5041.3  874.35  5065.5  876.45  5108.9  878.53  5136.7  882.44  5150.0  885.76
  5168.2  891.21  5179.8  893.94  5189.2  897.82  5206.2  903.24  5220.5  906.11
#Mann=3,-1,0
  4693.7    0.12       0  4975.3    0.04       0  5024.7    0.12       0
Bank Sta=4975.3,5024.7
XS Rating Curve= 0
Exp/Cntr=0.3,0.1

Type RM Length L Ch R = 1,49604,512,512,512
BEGIN DESCRIPTION:
North Hunting Creek 92.0
END DESCRIPTION:
XS GIS Cut Line= 4
      1468406.38       852587.12      1468304.90       852514.64
      1468155.81       852431.81      1468095.76       852384.19
#Sta/Elev= 30
  4742.7  897.20  4746.7  896.73  4770.3  890.13  4785.6  886.94  4812.1  882.21
  4824.8  880.26  4833.3  879.23  4861.1  876.15  4883.8  873.91  4886.5  873.82
  4909.6  874.84  4935.2  872.63  4943.1  872.27  4960.7  872.21  4966.0  871.01
  4970.8  869.11  4975.3  863.22  4976.3  861.22  5023.7  861.22  5024.7  863.22
  5028.2  863.27  5028.9  870.09  5034.7  875.79  5041.3  878.34  5053.2  884.80
  5062.3  888.11  5068.8  892.75  5087.3  907.90  5108.4  917.42  5114.6  919.82
#Mann=3,-1,0
  4742.7    0.12       0  4975.3    0.04       0  5024.7    0.12       0
#XS Ineff=2,0
    0.00 4909.60  874.84               0
Permanent Ineff=
       F       F
Bank Sta=4975.3,5024.7
XS Rating Curve= 0
Exp/Cntr=0.3,0.1

Type RM Length L Ch R = 1,49092,510,510,510
BEGIN DESCRIPTION:
North Hunting Creek 91.0
END DESCRIPTION:
XS GIS Cut Line= 4
      1468679.70       852175.07      1468580.29       852092.23
      1468408.43       851984.55      1468255.20       852021.82
#Sta/Elev= 30
  4754.0  891.74  4787.4  889.04  4806.6  885.58  4825.3  884.37  4840.6  881.36
  4846.9  878.92  4866.4  875.27  4906.0  872.69  4939.1  871.97  4958.6  869.60
  4958.9  865.77  4959.8  861.63  4975.3  861.63  4976.3  859.63  5023.7  859.63
  5024.7  861.63  5038.4  861.63  5042.3  868.46  5045.0  871.98  5078.1  875.06
  5094.0  876.92  5104.9  877.31  5110.6  878.22  5121.8  879.35  5150.1  884.56
  5171.5  890.24  5194.3  896.93  5205.8  900.67  5229.6  906.24  5243.9  907.48
#Mann=3,-1,0
  4754.0    0.12       0  4975.3    0.04       0  5024.7    0.12       0
Bank Sta=4975.3,5024.7
XS Rating Curve= 0
Exp/Cntr=0.3,0.1

Type RM Length L Ch R = 1,48582,608,608,608
BEGIN DESCRIPTION:
North Hunting Creek 90.0
END DESCRIPTION:
XS GIS Cut Line= 4
      1468729.38       851992.83      1468857.76       851758.85
      1468752.16       851524.87      1468669.32       851460.67
#Sta/Elev= 30
  4643.0  882.73  4724.9  882.60  4791.5  881.94  4795.4  881.76  4802.9  880.21
  4826.1  880.31  4867.8  876.95  4899.5  875.21  4913.6  873.63  4930.8  870.52
  4943.7  869.60  4966.9  862.55  4970.1  860.89  4975.3  860.86  4976.3  858.86
  5023.7  858.86  5024.7  860.86  5029.0  860.90  5029.5  863.89  5045.1  871.38
  5068.9  870.18  5082.7  870.17  5091.3  870.99  5144.6  871.77  5160.2  872.89
  5177.9  876.80  5214.6  888.65  5233.9  895.54  5241.2  898.59  5271.4  907.94
#Mann=3,-1,0
  4643.0    0.12       0  4975.3    0.04       0  5024.7    0.12       0
Bank Sta=4975.3,5024.7
XS Rating Curve= 0
Exp/Cntr=0.3,0.1

Type RM Length L Ch R = 1,47974,513,513,513
BEGIN DESCRIPTION:
North Hunting Creek 89.0
END DESCRIPTION:
XS GIS Cut Line= 4
      1469284.30       851796.15      1469338.15       851676.03
      1469234.62       851245.33      1469244.97       851129.40
#Sta/Elev= 30
  4451.1  892.31  4472.8  889.36  4515.7  881.71  4543.7  877.95  4582.7  875.84
  4686.7  872.29  4771.0  874.14  4812.3  873.92  4849.2  872.75  4880.3  870.26
  4895.0  868.18  4936.9  870.51  4953.8  869.51  4958.5  867.99  4961.4  863.55
  4967.8  858.37  4975.1  858.37  4976.1  856.37  5023.9  856.37  5024.9  858.37
  5034.6  858.37  5035.4  866.37  5038.0  867.91  5052.3  871.05  5058.6  874.78
  5070.2  884.57  5077.7  887.76  5098.4  895.03  5113.6  897.98  5142.1  901.05
#Mann=3,-1,0
  4451.1    0.12       0  4975.1    0.04       0  5024.9    0.12       0
#XS Ineff=2,0
    0.00 4936.90  870.51               0
Permanent Ineff=
       F       F
Bank Sta=4975.1,5024.9
XS Rating Curve= 0
Exp/Cntr=0.3,0.1

Type RM Length L Ch R = 1,47461,357,357,357
BEGIN DESCRIPTION:
North Hunting Creek 88.0
END DESCRIPTION:
XS GIS Cut Line= 4
      1470014.20       851531.06      1469954.17       851450.32
      1469695.34       851067.25      1469575.25       850984.44
#Sta/Elev= 30
  4482.7  895.25  4502.2  887.69  4539.6  876.29  4547.2  873.29  4562.9  870.64
  4572.5  871.47  4583.9  869.39  4604.7  867.53  4636.0  866.45  4647.0  864.34
  4667.9  866.26  4803.2  870.83  4847.4  870.37  4892.0  867.79  4904.3  867.01
  4920.4  867.20  4936.5  868.77  4946.9  868.64  4975.1  857.86  4976.1  855.86
  5023.9  855.86  5024.9  857.86  5027.4  858.11  5037.9  865.10  5051.8  870.60
  5079.9  874.60  5114.5  884.28  5123.9  888.39  5149.1  893.05  5191.5  895.22
#Mann=4,-1,0
  4482.7    0.06       0  4892.0    0.12       0  4975.1    0.04       0
  5024.9    0.12       0
#XS Ineff=2,0
    0.00 4821.90  870.39               0
Permanent Ineff=
       F       F
Bank Sta=4975.1,5024.9
XS Rating Curve= 0
Exp/Cntr=0.3,0.1

Type RM Length L Ch R = 1,47104,409,409,409
BEGIN DESCRIPTION:
North Hunting Creek 87.0
END DESCRIPTION:
XS GIS Cut Line= 4
      1470287.52       850914.03      1470181.94       850947.16
      1469911.99       850864.82      1469689.10       850911.96
#Sta/Elev= 30
  4707.4  896.85  4715.6  896.20  4727.1  892.95  4739.8  887.12  4759.9  880.58
  4785.5  871.10  4811.8  867.85  4822.3  867.27  4852.5  866.61  4894.4  867.58
  4912.0  867.27  4957.9  864.34  4961.4  862.43  4968.4  860.23  4975.1  855.24
  4976.1  853.24  5023.9  853.24  5024.9  855.24  5027.6  856.83  5044.6  861.83
  5063.3  865.91  5068.4  866.29  5079.7  865.42  5091.2  865.42  5110.9  867.02
  5150.9  868.51  5185.7  871.17  5253.0  878.12  5315.4  882.42  5328.1  882.66
#Mann=4,-1,0
  4707.4    0.06       0  4912.0    0.12       0  4975.1    0.04       0
  5024.9    0.12       0
#XS Ineff=2,0
    0.00 4894.40  867.58               0
Permanent Ineff=
       F       F
Bank Sta=4975.1,5024.9
XS Rating Curve= 0
Exp/Cntr=0.3,0.1

Type RM Length L Ch R = 1,46695,85,85,85
BEGIN DESCRIPTION:
North Hunting Creek 86.0
END DESCRIPTION:
XS GIS Cut Line= 4
      1469918.98       850514.37      1469869.27       850593.08
      1469792.66       850713.17      1469680.82       850901.64
#Sta/Elev= 30
  4902.0  895.65  4909.0  894.54  4910.1  893.96  4933.7  878.48  4945.1  869.90
  4962.6  864.07  4975.1  854.39  4976.1  852.39  5023.9  852.39  5024.9  854.39
  5025.4  856.83  5031.8  860.01  5040.4  862.18  5050.5  865.39  5056.4  865.88
  5067.9  865.70  5102.9  867.31  5120.1  867.57  5136.9  868.16  5155.8  868.38
  5167.5  869.01  5226.3  873.25  5244.0  875.04  5262.1  876.01  5275.1  877.52
  5291.3  878.52  5298.5  879.27  5316.5  880.15  5339.0  880.85  5356.7  881.93
#Mann=3,-1,0
  4902.0    0.12       0  4975.1    0.04       0  5024.9    0.08       0
Bank Sta=4975.1,5024.9
XS Rating Curve= 0
Exp/Cntr=0.5,0.3

Type RM Length L Ch R = 1,46610,42,42,42
BEGIN DESCRIPTION:
Sloans Mill Rd - US
END DESCRIPTION:
XS GIS Cut Line= 3
      1469931.37       850495.75      1469836.14       850477.12
      1469610.44       850880.89
#Sta/Elev= 30
  4821.2  896.69  4844.5  894.64  4853.6  893.24  4860.3  891.63  4885.6  888.42
  4903.8  885.11  4914.9  876.91  4918.2  875.62  4930.7  872.76  4933.6  872.71
  4950.2  868.65  4966.0  858.05  4969.5  857.50  4973.0  853.30  5027.0  853.30
  5030.5  857.50  5042.5  865.46  5044.6  866.22  5061.6  868.75  5108.4  869.73
  5140.4  869.64  5151.6  870.89  5167.7  870.93  5203.0  871.80  5238.8  873.19
  5264.9  875.09  5294.5  875.73  5312.8  878.24  5333.7  878.89  5380.8  883.80
#Mann=3,-1,0
  4821.2    0.08       0  4969.5    0.04       0  5030.5    0.08       0
#XS Ineff=2,0
    0.00 4933.00  872.90 5067.00    0.00  872.90
Permanent Ineff=
       F       F
Bank Sta=4969.5,5030.5
XS Rating Curve= 0
Exp/Cntr=0.5,0.3

Type RM Length L Ch R =3,46591,,,
BEGIN DESCRIPTION:
Sloans Mill Rd - TOR
Structure ID: LDS_NLHC_04
Approximate Survey Structure
END DESCRIPTION:
Bridge Culvert--1,0,-1,-1,0
Deck Dist Width WeirC Skew NumUp NumDn MinLoCord MaxHiCord MaxSubmerge Is_Ogee
9,20,3,,8,8,,,,0,1,1,,,
  4897.1  4919.9  4943.0  4943.0  5057.0  5057.0  5200.4  5234.8
  873.61  872.90  872.90  872.90  872.90  872.90  872.90  873.00
  833.30  833.30  833.30  871.40  871.40  833.30  833.30  833.30
  4897.1  4919.9  4943.0  4943.0  5057.0  5057.0  5200.4  5234.8
  873.61  872.90  872.90  872.90  872.90  872.90  872.90  873.00
  833.30  833.30  833.30  871.40  871.40  833.30  833.30  833.30
Pier Skew, UpSta & Num, DnSta & Num=,4962,2,4962,2,0,0,0,0,0
       1       1
  860.71  871.40
       1       1
  859.65  871.40
Pier Skew, UpSta & Num, DnSta & Num=,5000,2,5000,2,0,0,0,0,0
       1       1
  853.30  871.40
       1       1
  853.05  871.40
Pier Skew, UpSta & Num, DnSta & Num=,5038,2,5038,2,0,0,0,0,0
       1       1
  862.48  871.40
       1       1
  864.23  871.40
BR Coef=1,1,0,1.25,0,,,0.8,0,2,0,
WSPro=,,,, 1 ,,,, 0 ,,,, 0 ,,,,-1 ,-1 ,-1 , 0 , 0 , 0 , 0 , 0
BC Design=,,0,,0,,,,,,

Type RM Length L Ch R = 1,46568,419,419,419
BEGIN DESCRIPTION:
Sloans Mill Rd - DS
END DESCRIPTION:
XS GIS Cut Line= 3
      1469952.12       850475.05      1469809.22       850441.92
      1469573.15       850851.93
#Sta/Elev= 30
  4757.0  894.92  4791.5  893.10  4823.1  889.43  4833.3  889.00  4843.7  887.93
  4854.7  882.44  4865.4  874.24  4897.2  873.59  4903.7  873.88  4907.7  873.55
  4922.7  873.37  4932.6  872.72  4937.6  871.47  4950.1  867.20  4952.8  865.15
  4969.5  857.25  4973.0  853.05  5027.0  853.05  5030.5  857.25  5036.8  863.66
  5038.7  864.56  5056.3  870.20  5058.6  870.44  5074.7  870.97  5137.3  871.07
  5185.6  871.99  5246.8  873.97  5286.6  875.87  5335.7  880.53  5376.8  883.65
#Mann=3,-1,0
  4757.0    0.08       0  4969.5    0.04       0  5030.5    0.08       0
#XS Ineff=2,0
    0.00 4933.00  872.00 5067.00    0.00  872.00
Permanent Ineff=
       F       F
Bank Sta=4969.5,5030.5
XS Rating Curve= 0
Exp/Cntr=0.5,0.3

Type RM Length L Ch R = 1,46149,290,290,290
BEGIN DESCRIPTION:
North Little Hunting Creek 85.5
END DESCRIPTION:
XS GIS Cut Line= 4
      1469915.56       850426.77      1469748.28       850283.39
      1469668.63       850193.78      1469606.93       850092.27
#Sta/Elev= 30
  4681.4  887.58  4694.3  885.44  4696.3  884.27  4703.9  882.48  4714.2  878.66
  4724.1  877.23  4753.7  878.66  4760.3  879.92  4773.9  879.50  4839.7  871.33
  4859.6  868.17  4882.9  866.67  4904.3  863.04  4937.7  862.78  4956.1  861.28
  4958.8  853.33  4975.1  853.32  4976.1  851.32  5023.9  851.32  5024.9  853.32
  5027.8  853.35  5030.0  855.73  5039.3  863.36  5046.6  871.42  5067.1  881.02
  5072.0  882.71  5087.2  891.80  5114.7  903.70  5124.7  907.08  5140.4  911.12
#Mann=3,-1,0
  4681.4    0.12       0  4975.1    0.04       0  5024.9    0.12       0
Bank Sta=4975.1,5024.9
XS Rating Curve= 0
Exp/Cntr=0.3,0.1

Type RM Length L Ch R = 1,45859,503,503,503
BEGIN DESCRIPTION:
North Hunting Creek 85.0
END DESCRIPTION:
XS GIS Cut Line= 4
      1469974.88       850431.58      1469954.17       850299.04
      1469960.38       850104.40      1469939.68       850011.26
#Sta/Elev= 30
  4708.6  887.04  4716.5  885.15  4727.8  884.64  4742.0  881.06  4755.5  880.15
  4775.6  881.27  4784.0  881.32  4807.4  875.49  4822.2  873.15  4836.1  870.44
  4866.6  865.93  4878.7  864.47  4901.6  863.21  4918.3  863.21  4945.0  862.56
  4959.6  862.83  4960.7  859.87  4962.0  852.56  4975.0  852.56  4976.0  850.56
  5024.0  850.56  5025.0  852.56  5033.2  852.81  5052.1  866.07  5072.7  881.07
  5078.7  883.21  5094.0  891.30  5103.6  893.98  5128.0  907.75  5132.9  910.11
#Mann=3,-1,0
  4708.6    0.07       0  4975.0    0.04       0  5025.0    0.12       0
Bank Sta=4975,5025
XS Rating Curve= 0
Exp/Cntr=0.3,0.1

Type RM Length L Ch R = 1,45356,194,194,194
BEGIN DESCRIPTION:
North Little Hunting Creek 84.5
END DESCRIPTION:
XS GIS Cut Line= 3
      1470158.45       850611.97      1470242.12       850558.19
      1470415.35       850359.06
#Sta/Elev= 30
  4775.9  885.80  4780.6  884.22  4820.2  877.35  4836.9  873.60  4851.3  868.63
  4866.4  866.01  4882.1  865.34  4898.9  859.75  4916.7  852.89  4929.7  850.25
  4934.6  850.98  4952.7  847.91  4960.7  847.35  4968.3  844.88  4968.4  843.30
  4975.0  843.30  4976.0  841.30  5024.0  841.30  5025.0  843.30  5027.0  850.59
  5040.2  851.87  5051.7  855.07  5058.6  856.27  5068.2  859.92  5075.9  861.27
  5081.5  865.02  5093.6  870.71  5100.6  873.56  5110.5  876.27  5139.3  891.48
#Mann=3,-1,0
  4775.9    0.07       0  4975.0    0.04       0  5025.0    0.12       0
Bank Sta=4975,5025
XS Rating Curve= 0
Exp/Cntr=0.3,0.1

Type RM Length L Ch R = 1,45162,543,543,543
BEGIN DESCRIPTION:
North Hunting Creek 84.0
END DESCRIPTION:
XS GIS Cut Line= 4
      1470326.87       850760.82      1470405.57       850661.41
      1470511.17       850547.52      1470579.49       850475.06
#Sta/Elev= 30
  4783.2  888.38  4804.4  883.92  4821.4  880.89  4828.4  878.98  4834.7  874.72
  4845.8  867.74  4856.9  863.04  4873.7  863.26  4890.3  859.51  4907.9  851.59
  4922.0  849.27  4953.7  845.67  4966.7  843.51  4968.2  843.06  4969.6  841.36
  4975.0  841.36  4976.0  839.36  5024.0  839.36  5025.0  841.36  5033.7  841.42
  5036.4  841.70  5046.2  844.00  5062.0  846.50  5078.2  848.59  5085.2  851.92
  5091.7  855.57  5095.5  858.03  5108.2  867.64  5159.8  904.59  5164.9  906.70
#Mann=3,-1,0
  4783.2    0.07       0  4975.0    0.04       0  5025.0    0.12       0
Bank Sta=4975,5025
XS Rating Curve= 0
Exp/Cntr=0.3,0.1

Type RM Length L Ch R = 1,44619,585,585,585
BEGIN DESCRIPTION:
North Hunting Creek 83.0
END DESCRIPTION:
XS GIS Cut Line= 4
      1470612.60       851235.01      1470695.46       851150.08
      1470933.58       850882.97      1471022.64       850787.70
#Sta/Elev= 30
  4642.9  895.89  4655.2  892.59  4670.6  887.68  4696.8  876.40  4733.9  862.68
  4743.3  857.67  4755.3  853.84  4775.4  852.85  4789.5  852.97  4827.8  851.16
  4870.0  851.64  4896.4  851.79  4929.8  850.90  4946.4  847.29  4963.1  845.08
  4975.0  839.05  4976.0  837.05  5024.0  837.05  5025.0  839.05  5119.3  839.36
  5133.6  842.02  5149.3  848.83  5162.4  857.02  5175.8  861.69  5179.1  862.25
  5194.2  867.77  5212.5  883.14  5231.7  887.51  5241.8  890.72  5249.8  892.10
#Mann=4,-1,0
  4642.9    0.07       0  4870.0    0.12       0  4975.0    0.04       0
  5025.0    0.12       0
Bank Sta=4975,5025
XS Rating Curve= 0
Exp/Cntr=0.3,0.1

Type RM Length L Ch R = 1,44034,492,492,492
BEGIN DESCRIPTION:
North Hunting Creek 82.0
END DESCRIPTION:
XS GIS Cut Line= 4
      1471310.44       851473.12      1471329.08       851361.29
      1471358.07       851210.13      1471382.92       851065.14
#Sta/Elev= 30
  4800.5  882.79  4838.8  870.09  4843.7  868.04  4852.8  865.66  4864.6  857.09
  4876.7  854.14  4891.3  851.86  4905.9  850.59  4920.3  848.83  4937.3  849.63
  4951.3  845.93  4966.5  841.53  4972.8  838.23  4975.0  835.10  4976.0  833.10
  5024.0  833.10  5025.0  835.10  5029.1  838.48  5069.9  845.96  5081.0  850.39
  5082.7  850.50  5090.9  852.97  5108.8  864.74  5116.4  870.29  5126.8  872.56
  5152.3  876.57  5154.6  876.70  5164.9  878.58  5190.8  881.09  5214.9  882.66
#Mann=3,-1,0
  4800.5    0.12       0  4975.0    0.04       0  5025.0    0.12       0
Bank Sta=4975,5025
XS Rating Curve= 0
Exp/Cntr=0.3,0.1

Type RM Length L Ch R = 1,43542,296,296,296
BEGIN DESCRIPTION:
North Hunting Creek 81.0
END DESCRIPTION:
XS GIS Cut Line= 4
      1471888.16       851208.07      1471805.33       851145.94
      1471683.16       851065.18      1471587.87       851000.97
#Sta/Elev= 30
  4874.1  915.24  4886.2  908.50  4901.5  891.88  4932.2  871.03  4937.7  867.90
  4941.7  863.97  4944.5  858.37  4968.2  833.56  4975.0  833.56  4976.0  831.56
  5024.0  831.56  5025.0  833.56  5038.1  833.58  5039.5  835.74  5048.3  839.43
  5056.9  845.79  5059.6  845.93  5067.2  847.39  5074.6  847.87  5098.9  848.59
  5102.8  848.48  5108.2  848.91  5111.9  848.95  5129.1  850.57  5135.5  851.51
  5143.7  852.09  5163.7  857.93  5183.5  860.79  5192.4  861.79  5239.0  868.69
#Mann=3,-1,0
  4874.1    0.12       0  4975.0    0.04       0  5025.0    0.12       0
Bank Sta=4975,5025
XS Rating Curve= 0
Exp/Cntr=0.3,0.1

Type RM Length L Ch R = 1,43246,289,289,289
BEGIN DESCRIPTION:
North Little Hunting Creek 80.5
END DESCRIPTION:
XS GIS Cut Line= 4
      1472042.60       850950.07      1471955.99       850892.34
      1471827.53       850824.49      1471725.06       850752.33
#Sta/Elev= 30
  4888.3  893.36  4917.6  876.01  4932.7  865.25  4949.1  853.23  4965.2  843.00
  4975.0  833.22  4976.0  831.22  5024.0  831.22  5025.0  833.22  5027.7  833.23
  5047.5  839.90  5060.4  845.25  5076.8  844.00  5079.6  844.05  5082.3  843.49
  5094.1  844.84  5102.9  846.48  5114.5  847.27  5123.3  847.50  5131.1  847.45
  5143.7  848.56  5156.7  849.91  5195.7  862.91  5198.5  863.31  5216.8  864.82
  5225.0  866.07  5236.4  868.18  5244.7  869.45  5256.1  871.36  5263.0  871.94
#Mann=3,-1,0
  4888.3    0.12       0  4975.0    0.04       0  5025.0    0.12       0
Bank Sta=4975,5025
XS Rating Curve= 0
Exp/Cntr=0.3,0.1

Type RM Length L Ch R = 1,42957,441,441,441
BEGIN DESCRIPTION:
North Hunting Creek 80.0
END DESCRIPTION:
XS GIS Cut Line= 4
      1472167.68       850744.22      1472095.22       850648.98
      1471937.85       850568.23      1471832.28       850512.34
#Sta/Elev= 30
  4790.0  892.65  4815.1  884.17  4832.5  877.75  4843.2  874.32  4855.3  869.60
  4901.7  847.67  4910.2  844.21  4939.2  839.74  4947.4  838.95  4954.2  837.32
  4962.3  833.24  4972.1  830.44  4975.0  830.41  4976.0  828.41  5024.0  828.41
  5025.0  830.41  5027.5  830.41  5043.8  839.51  5048.2  843.84  5060.1  844.94
  5087.0  845.50  5105.5  848.72  5111.4  850.64  5129.8  857.72  5145.3  861.78
  5156.7  865.27  5182.9  869.70  5192.8  872.03  5197.1  872.04  5206.0  873.51
#Mann=3,-1,0
  4790.0    0.12       0  4975.0    0.04       0  5025.0    0.12       0
Bank Sta=4975,5025
XS Rating Curve= 0
Exp/Cntr=0.3,0.1

Type RM Length L Ch R = 1,42516,455,455,455
BEGIN DESCRIPTION:
North Hunting Creek 79.0
END DESCRIPTION:
XS GIS Cut Line= 4
      1472349.92       850427.45      1472285.72       850325.96
      1472217.38       850201.72      1472134.54       850141.67
#Sta/Elev= 30
  4767.8  869.59  4802.5  863.46  4820.5  858.52  4835.8  854.79  4849.0  852.30
  4860.7  848.70  4871.5  845.07  4882.6  842.38  4885.8  842.00  4897.2  841.20
  4910.2  839.81  4919.6  840.56  4933.7  842.56  4942.2  842.40  4952.5  840.80
  4956.2  839.09  4963.9  829.07  4975.0  829.07  4976.0  827.07  5024.0  827.07
  5025.0  829.07  5030.8  829.08  5035.6  834.38  5052.8  848.45  5066.4  860.88
  5086.1  871.70  5094.9  875.13  5108.0  879.58  5125.6  884.05  5132.0  885.21
#Mann=3,-1,0
  4767.8    0.12       0  4975.0    0.04       0  5025.0    0.12       0
#XS Ineff=2,0
    0.00 4933.70  842.56               0
Permanent Ineff=
       F       F
Bank Sta=4975,5025
XS Rating Curve= 0
Exp/Cntr=0.3,0.1

Type RM Length L Ch R = 1,42061,291,291,291
BEGIN DESCRIPTION:
North Hunting Creek 78.0
END DESCRIPTION:
XS GIS Cut Line= 4
      1472538.34       850450.20      1472637.73       850332.18
      1472646.01       850226.57      1472631.52       850137.56
#Sta/Elev= 30
  4763.4  861.75  4767.7  861.23  4782.7  859.95  4787.4  859.44  4818.5  855.52
  4835.6  852.19  4852.7  848.29  4859.6  847.13  4886.4  843.42  4918.0  839.69
  4921.2  839.45  4935.9  839.96  4939.2  839.93  4944.3  840.71  4957.3  842.37
  4962.2  842.08  4971.1  835.01  4975.0  828.14  4976.0  826.14  5024.0  826.14
  5025.0  828.14  5030.6  832.42  5044.5  839.37  5051.6  842.78  5057.7  846.96
  5064.3  852.96  5086.8  871.86  5092.0  877.55  5098.7  881.42  5113.8  891.35
#Mann=3,-1,0
  4763.4    0.12       0  4975.0    0.04       0  5025.0    0.12       0
Bank Sta=4975,5025
XS Rating Curve= 0
Exp/Cntr=0.3,0.1

Type RM Length L Ch R = 1,41770,238,238,238
BEGIN DESCRIPTION:
North Little Hunting Creek 77.5
END DESCRIPTION:
XS GIS Cut Line= 4
      1473046.44       850564.01      1472932.07       850411.53
      1472935.34       850230.68      1472940.79       850147.84
#Sta/Elev= 30
  4657.9  855.61  4726.0  849.29  4742.2  849.11  4747.6  848.76  4753.4  848.12
  4766.4  845.99  4795.2  843.90  4810.2  842.26  4832.4  840.72  4845.8  840.36
  4854.2  839.45  4873.5  838.09  4887.3  837.86  4900.8  836.93  4910.5  836.92
  4915.8  837.31  4926.1  837.17  4962.3  839.17  4967.3  839.01  4970.8  834.87
  4972.9  827.07  4973.9  825.07  5026.1  825.07  5027.1  827.07  5029.4  827.31
  5039.3  827.07  5043.3  827.25  5055.2  839.45  5059.3  841.87  5112.4  877.28
#Mann=3,-1,0
  4657.9    0.12       0  4972.9    0.04       0  5027.1    0.12       0
Bank Sta=4972.9,5027.1
XS Rating Curve= 0
Exp/Cntr=0.3,0.1

Type RM Length L Ch R = 1,41532,222,222,222
BEGIN DESCRIPTION:
North Hunting Creek 77.0
END DESCRIPTION:
XS GIS Cut Line= 4
      1473097.42       850557.84      1473147.10       850404.65
      1473171.95       850278.34      1473174.02       850170.63
#Sta/Elev= 30
  4738.0  855.92  4763.1  853.95  4773.0  852.81  4786.5  852.61  4800.1  851.71
  4840.5  847.39  4866.6  843.94  4878.3  842.63  4890.8  840.75  4903.5  840.26
  4915.9  839.30  4919.8  838.71  4929.1  838.94  4936.4  838.74  4941.9  836.82
  4958.5  826.13  4972.9  825.91  4973.9  823.91  5026.1  823.91  5027.1  825.91
  5032.9  825.91  5045.9  835.22  5052.8  839.55  5058.5  841.36  5087.4  853.62
  5089.9  855.51  5104.7  862.94  5125.0  873.64  5132.4  876.15  5135.5  876.80
#Mann=3,-1,0
  4738.0    0.12       0  4972.9    0.04       0  5027.1    0.12       0
Bank Sta=4972.9,5027.1
XS Rating Curve= 0
Exp/Cntr=0.5,0.3

Type RM Length L Ch R = 1,41310,39,39,39
BEGIN DESCRIPTION:
Hamptonville Rd - US
END DESCRIPTION:
XS GIS Cut Line= 5
      1473410.05       850752.47      1473331.39       850603.43
      1473325.18       850522.67      1473321.04       850491.62
      1473463.93       850073.30
#Sta/Elev= 30
  4520.0  856.88  4560.9  853.55  4616.6  850.93  4625.2  849.44  4635.8  849.72
  4646.7  848.35  4692.9  847.02  4702.4  844.34  4712.5  846.82  4729.9  844.65
  4741.2  845.33  4761.6  844.60  4797.9  844.96  4826.2  843.60  4909.8  845.07
  4924.0  846.45  4934.4  845.80  4951.4  840.94  4963.7  834.13  4969.0  834.10
  4980.0  823.60  5020.0  823.60  5031.0  831.59  5051.1  831.89  5080.8  847.12
  5092.7  847.64  5101.1  849.85  5203.9  857.12  5226.5  859.77  5242.9  859.87
#Mann=3,-1,0
  4520.0    0.12       0  4969.0    0.04       0  5031.0    0.12       0
#XS Ineff=2,0
    0.00 4924.50  849.00 5071.50    0.00  849.00
Permanent Ineff=
       F       F
Bank Sta=4969,5031
XS Rating Curve= 0
Exp/Cntr=0.5,0.3

Type RM Length L Ch R =3,41294,,,
BEGIN DESCRIPTION:
Hamptonville Rd - TOR
Structure ID: LDS_NLHC_03
Approximate Survey Structure
END DESCRIPTION:
Bridge Culvert--1,0,-1,-1,0
Deck Dist Width WeirC Skew NumUp NumDn MinLoCord MaxHiCord MaxSubmerge Is_Ogee
5.5,21,3,,8,8,,,,0,1,1,,,
  4636.8  4657.0  4934.5  4934.5  5065.5  5065.5  5083.9  5196.4
  849.64  849.00  849.00  849.00  849.00  849.00  849.00  855.52
  803.60  803.60  803.60  846.20  846.20  803.60  803.60  803.60
  4636.8  4657.0  4934.5  4934.5  5065.5  5065.5  5083.9  5196.4
  849.64  849.00  849.00  849.00  849.00  849.00  849.00  855.52
  803.60  803.60  803.60  846.20  846.20  803.60  803.60  803.60
Pier Skew, UpSta & Num, DnSta & Num=,4967.3,2,4967.3,2,0,0,0,0,0
       3       3
  834.11  846.20
       3       3
  834.38  846.20
Pier Skew, UpSta & Num, DnSta & Num=,5032.8,2,5032.8,2,0,0,0,0,0
       3       3
  830.42  846.20
       3       3
  825.92  846.20
BR Coef=1,1,0,1.25,0,,,0.8,0,2,0,
WSPro=,,,, 1 ,,,, 0 ,,,, 0 ,,,,-1 ,-1 ,-1 , 0 , 0 , 0 , 0 , 0
BC Design=,,0,,0,,,,,,

Type RM Length L Ch R = 1,41271,226,226,226
BEGIN DESCRIPTION:
Hamptonville Rd - DS
END DESCRIPTION:
XS GIS Cut Line= 4
      1473434.93       850727.68      1473360.38       850562.02
      1473356.24       850512.32      1473497.05       850075.39
#Sta/Elev= 30
  4574.9  857.67  4759.2  843.94  4841.8  842.86  4879.2  843.44  4886.4  841.94
  4898.7  841.43  4909.0  839.98  4935.6  841.00  4943.6  838.47  4950.6  837.79
  4956.3  835.16  4964.7  835.20  4969.0  833.85  4980.0  823.35  5020.0  823.35
  5031.0  828.98  5041.3  828.52  5052.5  829.84  5081.2  842.16  5093.7  844.21
  5114.9  851.31  5135.7  851.30  5160.8  854.71  5166.7  854.04  5190.4  855.19
  5208.5  856.68  5221.1  858.88  5242.4  859.05  5254.3  860.65  5265.5  860.85
#Mann=3,-1,0
  4574.9    0.12       0  4969.0    0.04       0  5031.0    0.12       0
#XS Ineff=2,0
    0.00 4924.50  847.65 5075.50    0.00  847.65
Permanent Ineff=
       F       F
Bank Sta=4969,5031
XS Rating Curve= 0
Exp/Cntr=0.5,0.3

Type RM Length L Ch R = 1,41045,478,478,478
BEGIN DESCRIPTION:
North Hunting Creek 76.0
END DESCRIPTION:
XS GIS Cut Line= 4
      1473526.05       850671.73      1473577.80       850537.17
      1473615.07       850317.68      1473631.64       850166.48
#Sta/Elev= 30
  4767.6  857.48  4801.3  852.07  4819.8  851.01  4842.5  848.59  4849.9  847.30
  4875.4  845.07  4909.7  841.42  4933.9  838.35  4948.5  837.38  4961.9  837.26
  4967.9  836.33  4970.1  833.29  4972.9  822.28  4973.9  820.28  5026.1  820.28
  5027.1  822.28  5029.0  825.56  5040.4  829.35  5056.5  838.47  5076.2  838.89
  5088.0  837.21  5122.0  838.20  5142.7  840.90  5148.6  842.12  5181.2  846.64
  5194.3  848.77  5205.7  851.46  5214.2  852.77  5247.4  855.34  5286.5  859.13
#Mann=3,-1,0
  4767.6    0.12       0  4972.9    0.04       0  5027.1    0.12       0
Bank Sta=4972.9,5027.1
XS Rating Curve= 0
Exp/Cntr=0.3,0.1

Type RM Length L Ch R = 1,40567,426,426,426
BEGIN DESCRIPTION:
North Hunting Creek 75.0
END DESCRIPTION:
XS GIS Cut Line= 4
      1474141.02       850410.87      1474056.12       850301.12
      1473923.60       850176.88      1473813.84       850046.41
#Sta/Elev= 30
  4784.8  870.46  4802.5  867.33  4810.2  867.33  4825.8  865.16  4851.2  859.90
  4898.6  846.30  4915.0  842.22  4923.6  839.41  4947.7  834.95  4959.4  835.65
  4961.7  833.17  4970.6  826.72  4972.9  821.39  4973.9  819.39  5026.1  819.39
  5027.1  821.39  5028.5  821.42  5030.3  824.03  5047.6  829.85  5063.5  835.95
  5069.2  835.97  5088.7  838.21  5103.8  841.67  5106.1  841.42  5143.0  843.72
  5150.0  846.60  5166.4  849.66  5226.1  854.87  5245.9  855.14  5275.7  857.09
#Mann=3,-1,0
  4784.8    0.12       0  4972.9    0.04       0  5027.1    0.12       0
Bank Sta=4972.9,5027.1
XS Rating Curve= 0
Exp/Cntr=0.3,0.1

Type RM Length L Ch R = 1,40141,663,663,663
BEGIN DESCRIPTION:
North Hunting Creek 74.0
END DESCRIPTION:
XS GIS Cut Line= 4
      1474447.47       850344.59      1474482.67       850176.88
      1474047.84       849619.87      1473942.27       849539.15
#Sta/Elev= 30
  4615.8  866.28  4644.9  862.52  4684.1  855.58  4697.0  854.55  4706.1  851.77
  4750.4  843.50  4779.4  839.74  4808.9  839.86  4917.3  834.72  4938.9  836.03
  4960.1  829.73  4972.9  821.02  4973.9  819.02  5026.1  819.02  5027.1  821.02
  5031.2  821.02  5031.9  823.64  5045.4  835.58  5072.4  834.41  5089.2  835.46
  5111.6  834.37  5141.2  834.88  5163.3  833.70  5213.1  835.43  5264.9  835.22
  5308.4  836.66  5416.3  836.19  5486.2  838.11  5567.7  860.74  5626.7  866.08
#Mann=3,-1,0
  4615.8    0.12       0  4972.9    0.04       0  5027.1    0.12       0
Bank Sta=4972.9,5027.1
XS Rating Curve= 0
Exp/Cntr=0.3,0.1

Type RM Length L Ch R = 1,39478,785,785,785
BEGIN DESCRIPTION:
North Hunting Creek 73.0
END DESCRIPTION:
XS GIS Cut Line= 4
      1475267.76       850075.30      1475203.19       849780.13
      1474259.20       849325.05      1474091.28       849371.41
#Sta/Elev= 30
  4335.5  850.99  4574.2  834.50  4652.8  830.89  4770.1  833.99  4820.1  833.47
  4893.2  834.51  4922.1  836.47  4956.4  836.01  4968.0  834.48  4970.6  829.06
  4972.3  820.47  4972.9  820.46  4973.9  818.46  5026.1  818.46  5027.1  820.46
  5034.4  820.47  5034.7  829.96  5036.1  833.34  5058.2  836.18  5419.6  834.47
  5643.4  831.82  5699.8  833.35  5710.8  834.44  5718.5  837.59  5728.9  838.19
  5750.9  842.92  5768.2  844.28  5776.3  848.25  5800.5  854.21  5859.8  861.92
#Mann=3,-1,0
  4335.5    0.09       0  4972.9    0.04       0  5027.1    0.07       0
#XS Ineff=2,0
    0.00 4933.90  836.64 5058.20    0.00  836.18
Permanent Ineff=
       F       F
Bank Sta=4972.9,5027.1
XS Rating Curve= 0
Exp/Cntr=0.3,0.1

Type RM Length L Ch R = 1,38693,787,787,787
BEGIN DESCRIPTION:
North Hunting Creek 72.0
END DESCRIPTION:
XS GIS Cut Line= 4
      1475464.53       848817.71      1475190.89       848983.74
      1474185.41       849217.43      1474064.39       849321.71
#Sta/Elev= 30
  4553.1  884.60  4600.5  871.77  4626.9  861.29  4667.0  849.09  4687.5  845.43
  4704.5  840.46  4752.3  830.62  4757.0  831.01  4765.8  835.14  4848.8  846.26
  4875.5  847.25  4894.6  846.21  4916.2  843.06  4943.4  833.18  4963.2  822.39
  4972.9  819.78  4973.9  817.78  5026.1  817.78  5027.1  819.78  5034.9  832.20
  5054.7  833.77  5099.2  832.55  5188.3  834.42  5487.7  830.99  5877.3  832.49
  5896.5  834.11  5912.3  838.84  5956.3  847.51  5974.9  853.03  6065.2  862.24
#Mann=3,-1,0
  4553.1    0.12       0  4972.9    0.04       0  5027.1    0.07       0
#XS Ineff=2,0
    0.00 4865.60  847.06 5054.70    0.00  833.77
Permanent Ineff=
       F       F
Bank Sta=4972.9,5027.1
XS Rating Curve= 0
Exp/Cntr=0.3,0.1

Type RM Length L Ch R = 1,37906,688,688,688
BEGIN DESCRIPTION:
North Hunting Creek 71.0
END DESCRIPTION:
XS GIS Cut Line= 5
      1475169.37       847929.06      1475095.57       847981.33
      1474420.55       848559.70      1474431.40       848814.62
      1474016.26       849251.28
#Sta/Elev= 30
  4343.0  853.76  4373.6  846.35  4415.4  829.55  4442.5  826.46  4530.7  829.67
  4678.8  828.93  4902.0  832.13  4954.7  833.23  4971.5  828.57  4972.9  818.89
  4973.9  816.89  5026.1  816.89  5027.1  818.89  5030.9  818.89  5032.4  822.85
  5034.8  824.74  5063.8  830.55  5123.3  829.65  5176.3  832.09  5257.3  829.03
  5322.3  834.02  5371.0  841.22  5406.5  843.24  5602.4  840.17  5744.2  833.37
  5899.9  836.12  6005.8  841.06  6053.8  848.58  6091.6  850.61  6180.0  859.32
#Mann=4,-1,0
  4343.0    0.07       0  4902.0    0.12       0  4972.9    0.04       0
  5027.1    0.07       0
#XS Ineff=2,0
    0.00 4951.40  833.27               0
Permanent Ineff=
       F       F
Bank Sta=4972.9,5027.1
XS Rating Curve= 0
Exp/Cntr=0.3,0.1

Type RM Length L Ch R = 1,37218,636,636,636
BEGIN DESCRIPTION:
North Hunting Creek 70.0
END DESCRIPTION:
XS GIS Cut Line= 4
      1475045.87       847700.39      1474952.71       847741.80
      1474225.91       847863.96      1474128.63       847849.47
#Sta/Elev= 30
  4350.3  857.61  4353.0  857.44  4382.9  847.03  4418.7  832.34  4431.3  829.29
  4443.5  829.15  4466.6  826.42  4508.7  827.95  4816.3  829.23  4909.7  831.14
  4921.7  830.96  4934.9  823.57  4947.0  821.92  4961.9  818.39  4972.9  817.61
  4973.9  815.61  5026.1  815.61  5027.1  817.61  5028.3  826.11  5032.7  826.08
  5042.1  829.74  5096.6  826.25  5126.7  827.19  5164.7  826.77  5174.5  825.10
  5187.1  829.89  5204.3  832.45  5231.5  841.12  5249.8  848.26  5287.6  859.33
#Mann=4,-1,0
  4350.3    0.07       0  4947.0    0.12       0  4972.9    0.04       0
  5027.1    0.12       0
Bank Sta=4972.9,5027.1
XS Rating Curve= 0
Exp/Cntr=0.3,0.1

Type RM Length L Ch R = 1,36582,582,582,582
BEGIN DESCRIPTION:
North Hunting Creek 69.0
END DESCRIPTION:
XS GIS Cut Line= 4
      1475054.18       847658.98      1474981.70       847582.36
      1474203.13       847263.48      1474082.99       847275.91
#Sta/Elev= 30
  4160.2  858.26  4168.3  857.46  4228.2  836.13  4250.0  830.20  4279.7  826.40
  4371.4  828.37  4452.6  828.15  4498.9  829.08  4712.4  827.97  4744.7  827.12
  4770.0  828.23  4794.6  829.19  4882.6  828.77  4925.6  830.47  4947.9  830.03
  4961.7  823.50  4962.8  822.45  4964.2  817.17  4972.8  817.17  4973.8  815.17
  5026.2  815.17  5027.2  817.17  5031.8  817.22  5035.6  827.96  5036.5  828.99
  5055.9  830.09  5096.0  828.93  5115.7  830.06  5153.5  839.63  5227.8  851.21
#Mann=4,-1,0
  4160.2    0.07       0  4770.0    0.12       0  4972.8    0.04       0
  5027.2    0.12       0
Bank Sta=4972.8,5027.2
XS Rating Curve= 0
Exp/Cntr=0.3,0.1
